HEC-RAS study THRNYCK.prj: THRNYCK

--- THRNYCK.g01 (geometry) --- (continued)

Type RM Length L Ch R = 1 ,43703   ,304.1,288.9,269.2
XS GIS Cut Line= 4
2268723.36460932466291.2402184042268581.13692941466504.120040716
2268549.44156416466685.2106541582268568.89502885466743.571048218
#Sta/Elev= 30
       0 2618.18     9.5 2615.26    16.8  2613.7    31.2 2609.16    55.2 2603.03
    69.7 2598.18    72.9 2596.44    75.8 2594.43    84.4 2586.59    87.3 2585.24
    88.9 2584.88    98.5 2584.78   113.7 2584.97   119.1 2585.39   132.2  2588.3
     137 2588.73   156.5 2588.81   175.5 2588.25   185.1 2588.47   209.2 2587.77
   237.3 2587.44   257.1 2588.06   293.6 2587.13   326.1 2587.84   350.5  2588.9
   385.6 2589.22   395.2 2589.01   407.3 2590.62   448.5 2590.94   501.4  2592.3
#Mann= 4 ,-1,0
       0      .1       0    87.3    .045       0   119.1      .1       0
     200     .05       0
#XS Ineff= 2 , 0
                          327.11          2600.7
Permanent Ineff=
       F       F
Bank Sta=87.3,119.1
XS Rating Curve= 0 ,0
Exp/Cntr(USF)=0,0
Exp/Cntr=0.3,0.1

Type RM Length L Ch R = 1 ,43414   ,316.2,313.3,305.2
XS GIS Cut Line= 3
2268389.06978661466252.8558009832268424.30318473466489.488615321
2268401.90260959466726.614481182
#Sta/Elev= 30
       0  2607.5    17.1  2602.8      30 2599.71    38.2 2596.27    52.9  2587.7
    56.9 2586.11      65  2584.3    73.1 2583.47    80.5 2583.67    85.3 2584.17
    89.3 2584.27    97.4 2583.47   101.6  2583.8   105.5 2584.73   109.5 2585.13
   113.6 2584.95   121.6 2585.35   133.8 2584.82   137.8 2584.31   145.9 2584.24
     154 2585.81     158 2587.08   162.1 2587.21   182.3 2586.78   194.4 2587.37
   222.8 2587.97   267.1 2588.23   319.8 2589.24   391.6 2589.17   477.4 2591.33
#Mann= 5 ,-1,0
       0      .1       0      65    .045       0    85.3      .1       0
     110     .05       0  399.24     .06       0
Bank Sta=65,85.3
XS Rating Curve= 0 ,0
Exp/Cntr(USF)=0,0
Exp/Cntr=0.3,0.1

Type RM Length L Ch R = 1 ,43101   ,137.5,149.6,160.9
XS GIS Cut Line= 3
2268109.74726351466326.1929568262268105.95403764466400.453994532
2268251.69692874466734.538952399
#Sta/Elev= 30
       0 2603.84      11 2600.99      15 2600.27      27 2597.43      35 2596.04
      47 2594.39    71.1    2592    76.6 2591.27    79.5  2590.7    88.2 2587.51
    92.6 2586.41      97 2585.91   105.7 2585.62   136.2 2585.45   143.4 2585.17
     145 2585.05   153.7 2583.26   159.9  2582.6   170.8 2582.16   175.5 2582.19
   179.9 2582.53   188.6 2584.75     193 2585.21   232.3 2586.09   261.9 2587.84
   319.7 2587.81     344 2588.41   376.3  2588.7   402.5 2589.15   438.8 2590.07
#Mann= 4 ,-1,0
       0      .1       0  134.36     .05       0   159.9    .045       0
   179.9     .05       0
Bank Sta=159.9,179.9
XS Rating Curve= 0 ,0
Exp/Cntr(USF)=0,0
Exp/Cntr=0.3,0.1

Type RM Length L Ch R = 1 ,42951   ,237,241.6,245.5
XS GIS Cut Line= 4
2268000.17859255466340.2995943252268013.54584236466403.022843443
2267976.26391817466613.1424710472268025.06143811466790.835225147
#Sta/Elev= 30
       0 2607.44     9.1 2603.45    17.6 2600.34    27.7 2597.55    41.8 2594.48
    65.1 2591.65    78.5 2589.49   106.9 2587.25   131.3 2585.95   135.4  2585.4
   143.5 2582.33   151.6 2581.86   163.8 2582.15   171.9 2583.02   180.1 2584.22
   184.1 2584.33   208.5 2582.81     219 2583.06   239.7 2583.09   257.3 2582.66
   269.4 2583.23   273.5 2584.33   277.5    2585   298.3 2586.33   313.3 2586.91
   348.1 2587.75   377.1 2589.34   393.7 2589.74   443.5 2589.59   461.8 2589.94
#Mann= 4 ,-1,0
       0      .1       0   143.5    .045       0   163.8      .1       0
  214.13     .05       0
Bank Sta=143.5,163.8
XS Rating Curve= 0 ,0
Exp/Cntr(USF)=0,0
Exp/Cntr=0.3,0.1

Type RM Length L Ch R = 1 ,42710   ,245.5,233.3,217.8
XS GIS Cut Line= 4
2267791.93907772466324.6367824672267792.97378314466370.830635539
2267743.21247157466490.5413556252267777.04834568466815.351087644
#Sta/Elev= 30
       0  2612.4     8.5 2609.91    20.5 2605.73    36.6 2600.93    40.6 2599.34
    44.6 2597.11    48.6 2593.87    54.7 2589.33    61.7 2584.66    63.9 2583.71
    66.1 2582.95    74.7 2581.79    79.2 2581.31 89.84292580.894    97.6  2580.8
108.3316 2580.86   113.7  2580.9   118.1  2581.2   125.1 2583.03   131.7 2583.59
   146.5 2583.66     157 2584.08   173.3 2583.99   238.8  2584.6   287.1 2586.03
   366.3 2586.59   387.6 2586.43   403.7    2587     452    2588   502.4 2588.73
#Mann= 6 ,-1,0
       0      .1       0      30     .05       0 89.8429    .045       0
108.3316     .05       0  126.21      .1       0  136.21     .05       0
Bank Sta=89.8429,108.3316
XS Rating Curve= 0 ,0
Exp/Cntr(USF)=0,0
Exp/Cntr=0.3,0.1

Type RM Length L Ch R = 1 ,42476   ,197.9,201.6,204.4
XS GIS Cut Line= 2
2267530.26834915466360.8645940362267701.98609674466828.718337456
#Sta/Elev= 30
       0 2620.38     4.8 2618.08    11.1 2615.79    17.3 2612.89    26.7 2607.79
    29.8 2605.78    42.3  2595.9    51.6 2586.73    55.7 2583.86      60 2582.48
    66.82581.543    76.5 2580.47    81.92581.382    85.9 2582.33    89.8  2582.8
   101.5 2582.03     110 2582.72   123.9 2582.58   138.9 2583.91   145.2 2585.32
   148.2 2585.44   179.3 2585.06   238.9 2585.91     273 2585.09     301 2585.05
   336.9 2585.56   385.1 2587.48   423.5 2588.01   456.3 2587.87   498.4 2588.74
#Mann= 4 ,-1,0
       0      .1       0    66.8    .045       0    81.9      .1       0
     110     .05       0
Bank Sta=66.8,81.9
XS Rating Curve= 0 ,0
Exp/Cntr(USF)=0,0
Exp/Cntr=0.3,0.1

Type RM Length L Ch R = 1 ,42275   ,141.2,142.5,143.2
XS GIS Cut Line= 2
2267373.97435135466421.5313431832267466.51685005466862.650586979
#Sta/Elev= 30
       0 2614.07      16 2604.38    32.3 2595.27    40.5 2589.94    44.6 2587.85
    48.7 2586.41    56.9 2584.79    75.9 2582.94    81.4 2582.76    93.6 2580.65
   105.9 2580.23   114.1 2580.25   123.2 2579.54   130.4 2579.04   138.6 2579.25
   140.1 2579.59   142.7 2580.31   146.8 2582.08   160.3 2584.08   175.4 2583.84
   220.3 2584.27   236.7 2584.01   269.4 2584.32   295.5 2584.18     309  2584.6
     347 2584.97   376.6 2585.78   405.3  2586.2   432.9 2587.52   450.7 2587.74
#Mann= 3 ,-1,0
       0      .1       0   123.2    .045       0   140.1     .05       0
#XS Ineff= 2 , 0
                          295.18          2597.2
Permanent Ineff=
       F       F
Bank Sta=123.2,140.1
XS Rating Curve= 0 ,0
Exp/Cntr(USF)=0,0
Exp/Cntr=0.3,0.1

Type RM Length L Ch R = 1 ,42132   ,105,104.8,106.7
XS GIS Cut Line= 3
2267242.50526295466453.5573993232267284.56776437466710.076975339
2267330.82409437466844.483540744
#Sta/Elev= 30
       0 2617.15     7.7  2613.2    15.1 2608.54    19.9 2604.97      28 2598.22
    42.9 2587.36    48.3 2584.68    52.3 2583.46    56.4 2582.99    64.5 2582.96
    74.3 2581.76   105.6 2581.93   109.1 2581.63   117.2 2579.97   129.3 2578.93
   133.4 2578.81   145.5 2579.01   148.52579.435   153.6 2580.99   161.8 2581.04
     178  2582.8   189.2 2582.89   194.2 2582.49   206.3 2582.37   246.9 2584.97
   267.5 2585.75   335.1 2585.57   356.5 2585.84   381.7 2586.69   402.1 2586.66
#Mann= 5 ,-1,0
       0      .1       0     100     .05       0   129.3    .045       0
   148.5     .05       0  402.09     .06       0
#XS Ineff= 2 , 0
                          286.48         2588.28
Permanent Ineff=
       F       F
Bank Sta=129.3,148.5
XS Rating Curve= 0 ,0
Exp/Cntr(USF)=0,0
Exp/Cntr=0.3,0.1

Type RM Length L Ch R = 1 ,42027   ,279.6,285.2,294.1
XS GIS Cut Line= 2
2267149.81585451466477.0568424022267187.86110397466880.130836733
#Sta/Elev= 30
       0 2610.39    16.2 2603.16    20.2 2600.94    32.3 2593.79    44.3 2585.28
    48.3  2583.1    52.4 2582.32    60.4 2581.91    64.4 2581.14    68.5 2581.48
    84.5 2579.19    92.5 2579.17    96.5 2579.48   104.6 2580.86   108.7    2581
   120.7 2580.59   134.4 2578.97   140.7 2578.62   148.4 2579.08   152.8 2580.66
   160.8 2582.41   164.9 2582.88   195.4 2582.51     209 2581.94   229.9 2581.86
   241.2 2582.34   257.3 2583.93   269.3 2584.66   353.7 2585.94   404.9 2587.32
#Mann= 5 ,-1,0
       0      .1       0   134.4    .045       0   148.4      .1       0
     270     .05       0     370     .06       0
Bank Sta=134.4,148.4
XS Rating Curve= 0 ,0
Exp/Cntr(USF)=0,0
Exp/Cntr=0.3,0.1

Type RM Length L Ch R = 1 ,41742   ,216.1,210.3,202.7
XS GIS Cut Line= 2
2266964.73085711466432.842093023  2266830.030109466773.192838237
#Sta/Elev= 30
       0 2621.23       9 2616.36    26.2 2602.57    39.1 2590.07    46.9 2584.78
      52 2580.87    53.1 2580.38    56.3 2579.75    64.9 2579.25    74.7 2578.11
    77.8 2577.87    88.5 2578.32    90.7 2578.64      95 2579.94    99.3 2580.66
   129.4 2580.74     138 2580.31   150.9 2579.06     164 2578.99   168.1 2579.21
   176.7 2580.45   185.3 2580.68   198.2 2581.56   241.1 2580.81   287.3 2581.94
   305.8 2583.94   327.4 2584.25   335.9 2584.99   344.5 2586.51     366 2592.69
#Mann= 4 ,-1,0
       0      .1       0    74.7    .045       0    88.5      .1       0
     240     .05       0
Bank Sta=74.7,88.5
XS Rating Curve= 0 ,0
Exp/Cntr(USF)=0,0
Exp/Cntr=0.3,0.1

Type RM Length L Ch R = 1 ,41532   ,177.3,179.5,179.8
XS GIS Cut Line= 3
2266741.60061025466381.429593747 2266737.4804055466547.862378277
2266671.57778874466706.362342614
#Sta/Elev= 30
       0 2618.55     3.8 2616.25    11.8 2610.28    18.8 2603.91    27.8 2596.39
    31.8 2592.46    36.3 2587.37    40.2 2583.83    43.8  2581.5    47.5 2579.72
    51.8 2578.81    55.8 2578.56    63.8 2579.18    79.8 2576.87    95.8 2576.56
     105 2576.86   111.8 2577.76   131.8 2578.43   139.8 2580.09   172.2 2580.56
   185.2 2580.07   189.6 2579.39   193.9 2579.25   199.1 2579.65   206.9 2581.31
   211.2 2581.69   248.1 2582.56   302.2 2585.09   323.9  2586.5   338.1 2586.61
#Mann= 5 ,-1,0
       0      .1       0    79.8    .045       0     105      .1       0
  276.48     .05       0  316.48      .1       0
Bank Sta=79.8,105
XS Rating Curve= 0 ,0
Exp/Cntr(USF)=0,0
Exp/Cntr=0.3,0.1

Type RM Length L Ch R = 1 ,41352   ,167.1,167.7,168.4
XS GIS Cut Line= 3
 2266588.3913624 466378.344843792266568.85461268 466417.41834324
2266559.60036281466644.661590044
#Sta/Elev= 30
       0 2615.27     7.6 2611.13    12.1 2609.03    18.4 2605.51    25.5 2601.26
      30 2598.25    34.5 2594.96    44.1 2587.49    47.4 2585.47    51.5 2583.38
    55.6 2580.92    59.5 2578.79    63.5 2577.84    82.6 2576.86    91.5 2576.47
    95.5 2576.81    99.5 2577.72   107.5 2578.93   119.5 2579.92   127.5 2580.06
   135.5 2580.54     148 2580.85   159.5 2581.53   175.6 2581.65   183.6    2582
   203.6 2583.75   243.6 2585.25   251.6 2585.77   255.7 2585.88   271.1 2587.07
#Mann= 3 ,-1,0
       0      .1       0    82.6    .045       0    95.5      .1       0
Bank Sta=82.6,95.5
XS Rating Curve= 0 ,0
Exp/Cntr(USF)=0,0
Exp/Cntr=0.3,0.1

Type RM Length L Ch R = 1 ,41185   ,314.4,342.3,358.1
XS GIS Cut Line= 3
2266473.22736402466290.9435950192266407.41936495466376.288343819
2266384.79786526 466636.43559016
#Sta/Elev= 30
       0 2615.47    13.8 2605.01    27.9 2593.01    34.5 2589.23    43.2 2582.46
    48.3 2579.49    53.3 2578.74    59.4 2578.73    68.5 2577.99    90.8 2579.17
   124.7 2578.88   136.8 2579.45   144.8 2579.25   156.8 2578.14   164.9 2576.26
   176.9 2576.04   180.9 2575.91     197 2575.95     201 2576.43     209 2579.11
   213.1 2579.41   217.1 2579.51   225.1  2578.7   245.9 2577.79   257.2 2578.66
   265.3 2581.16   274.1 2582.57   317.4 2584.25   361.6 2585.51   368.9  2585.4
#Mann= 5 ,-1,0
       0      .1       0      80     .12       0   176.9    .045       0
     197      .1       0  347.77     .12       0
Bank Sta=176.9,197
XS Rating Curve= 0 ,0
Exp/Cntr(USF)=0,0
Exp/Cntr=0.3,0.1

Type RM Length L Ch R = 1 ,40842   ,118.7,118.7,118.6
XS GIS Cut Line= 3
2266425.92786469466270.3785953082266268.90559343466413.134798354
2266063.68568111466416.368306012
#Sta/Elev= 30
       0  2603.7     6.1  2599.6    16.1 2591.66    20.2 2588.96    34.4 2580.88
    40.2 2579.38    57.7 2578.92    69.6 2577.64    93.8 2577.84   110.5 2575.85
     125 2576.15   153.3 2578.87   164.7 2578.53   176.6 2577.33   190.1 2577.39
   202.4 2578.79   224.9 2577.61     245 2577.17     269 2577.35     277 2575.26
     285  2574.8   287.8  2575.2     301 2575.95   314.5 2574.79     317 2574.81
     333 2580.29     337 2581.06     357  2582.4   399.9 2583.85   417.5 2584.92
#Mann= 6 ,-1,0
       0      .1       0      60     .12       0     190      .1       0
     277    .045       0   287.8      .1       0  392.22     .05       0
Bank Sta=277,287.8
XS Rating Curve= 0 ,0
Exp/Cntr(USF)=0,0
Exp/Cntr=0.3,0.1

Type RM Length L Ch R = 1 ,40724   ,235.2,230.9,226.7
XS GIS Cut Line= 3
2266391.99561516466222.0508459882266277.85986677466294.028344976
 2266019.7691204 466302.25434486
#Sta/Elev= 30
       0  2604.7    25.3 2587.23    37.6 2579.55    42.3 2577.17    43.4 2576.98
    50.9 2576.77    65.9 2577.78    77.5 2578.02    84.9 2577.28    94.4 2574.86
   108.6  2575.5     118 2574.99   137.6 2577.57   155.1 2577.96   180.6 2577.31
   208.7 2574.93   220.7 2574.22   228.8 2574.61   232.7 2574.72   240.7 2576.26
   268.7 2577.14   300.7 2579.13   308.7 2579.27   316.7 2580.12   328.7  2579.8
   352.7  2580.7   360.8 2580.38   373.2 2582.23   384.7 2584.82   393.2 2586.28
#Mann= 6 ,-1,0
       0      .1       0      60     .12       0     130      .1       0
   208.7    .045       0   228.8      .1       0  324.94     .05       0
Bank Sta=208.7,228.8
XS Rating Curve= 0 ,0
Exp/Cntr(USF)=0,0
Exp/Cntr=0.3,0.1

Type RM Length L Ch R = 1 ,40493   ,412.5,417.1,412.1
XS GIS Cut Line= 2
2266304.59436639466046.2200984612265921.05712179466142.875597102
#Sta/Elev= 30
       0 2612.88     4.6 2610.55      16 2603.54    25.8 2596.52    33.4 2591.77
    48.9 2581.28    58.2 2576.64    62.3 2575.58    70.6  2574.5    74.7 2574.09
    78.8 2574.44    87.1 2573.06    91.7  2573.3   111.8 2575.72   124.7 2576.28
   128.3 2576.31   136.6 2575.36   148.9 2575.06   165.4 2573.99   187.3 2574.02
   219.1 2574.61   235.6 2577.28   247.9 2579.73   252.1  2580.1   261.2 2579.95
   272.7 2580.66   293.3 2582.99   305.9 2583.85   330.4 2584.78   395.5 2585.88
#Mann= 4 ,-1,0
       0      .1       0   165.4    .045       0   187.3      .1       0
     220     .05       0
Bank Sta=165.4,187.3
XS Rating Curve= 0 ,0
Exp/Cntr(USF)=0,0
Exp/Cntr=0.3,0.1

Type RM Length L Ch R = 1 ,40076   ,168.5,180.6,193.2
XS GIS Cut Line= 2
2266271.35368651465797.561626905 2265857.8810232465927.661090013
#Sta/Elev= 30
       0 2610.35    15.9 2602.36    20.1 2600.52    25.4  2597.5    45.3 2584.05
    49.5 2580.94    57.8 2574.05      62  2572.6    66.6 2571.39    70.4 2570.77
    74.6 2570.64      83 2571.04    91.4 2571.72   126.6 2572.87   137.5 2572.92
   145.9 2573.86   154.3 2574.51   171.1  2574.5   183.6 2573.67   187.2 2573.79
     192 2574.33   200.4 2576.33   209.6 2577.07   270.2 2577.21   301.1 2577.62
   340.3 2577.02     385 2577.31   401.7 2578.34   425.2 2581.45   433.5 2582.18
#Mann= 5 ,-1,0
       0      .1       0    66.6    .045       0      83      .1       0
      90     .08       0     190     .05       0
Bank Sta=66.6,83
XS Rating Curve= 0 ,0
Exp/Cntr(USF)=0,0
Exp/Cntr=0.3,0.1

Type RM Length L Ch R = 1 ,39895   ,149.2,147.8,147.5
XS GIS Cut Line= 4
2266279.75882682465739.0156573542266232.26670531465694.817633926
2266058.81570636465619.4720961952265884.79082499465628.725255782
#Sta/Elev= 30
       0 2608.75    20.3 2598.84    32.1 2591.99    43.1 2585.03    49.1 2582.22
    61.4 2579.81    73.7 2578.14    87.5 2574.93    95.5 2572.42   104.2  2570.7
   108.6 2570.37   120.9 2571.67   130.4 2571.73   145.2 2570.32   157.4 2569.68
   169.4 2569.25   172.6 2569.92   181.7 2573.11   187.1 2573.76   204.5 2571.69
   217.6 2572.11   233.4 2571.71   239.5 2572.33   248.1 2574.87   256.6 2574.94
   276.7 2574.12   292.7 2574.96   328.7 2575.47   360.7  2576.5   428.3 2577.39
#Mann= 6 ,-1,0
       0      .1       0  114.88     .08       0  154.88      .1       0
   157.4    .045       0   172.6      .1       0  224.88     .05       0
Bank Sta=157.4,172.6
XS Rating Curve= 0 ,0
Exp/Cntr(USF)=0,0
Exp/Cntr=0.3,0.1

Type RM Length L Ch R = 1 ,39747   ,273.9,267.9,257.4
XS GIS Cut Line= 4
2266336.41119288465556.4333893962266262.65656096465549.126046985
2266049.53124498465469.8402815682265855.30624771465470.982781551
#Sta/Elev= 30
       0 2614.06    16.3 2606.39    40.4 2596.19    56.5  2591.3    60.5 2589.26
      69 2583.86    72.7 2581.98    76.8 2578.89      81 2576.37    96.9  2570.8
106.91042568.433   110.9 2568.24121.38032568.412     128 2569.02   136.5 2570.42
   149.3 2570.91   162.1 2571.98   170.7 2571.28     192 2571.49   196.3 2571.76
   204.8 2573.12   217.6 2572.64   243.2 2573.41   285.9 2572.84   310.9 2573.47
   338.9 2573.38   354.9 2573.76   362.9 2574.88   382.9 2575.22   495.7 2575.62
#Mann= 4 ,-1,0
       0      .1       0106.9104    .045       0121.3803      .1       0
  154.12     .05       0
Bank Sta=106.9104,121.3803
XS Rating Curve= 0 ,0
Exp/Cntr(USF)=0,0
Exp/Cntr=0.3,0.1

Type RM Length L Ch R = 1 ,39479   ,247,252.5,256.2
XS GIS Cut Line= 2
2266386.82262913465281.0738953342265815.57263716465314.079450425
#Sta/Elev= 30
       0 2615.24     2.7 2614.62     6.7 2612.23    10.7 2609.22    14.7 2605.54
    34.7 2589.77    58.7 2573.96    62.8 2572.45    70.7 2570.54    78.4 2569.52
    86.8 2568.95    98.8 2568.56   106.8 2569.08   114.8 2571.77   118.8 2571.99
   146.5 2570.71   154.9 2570.62     199 2572.02   243.1 2572.92   263.1 2572.44
   300.4 2572.38   364.2 2573.59   423.4 2573.22   451.4 2574.44   467.4 2574.21
   476.1 2574.69   487.5 2574.09   502.6 2575.28   515.5 2575.71   572.2 2576.17
#Mann= 3 ,-1,0
       0      .1       0    86.8    .045       0   106.8     .05       0
#XS Ineff= 2 , 0
                          365.66         2586.85
Permanent Ineff=
       F       F
Bank Sta=86.8,106.8
XS Rating Curve= 0 ,0
Exp/Cntr(USF)=0,0
Exp/Cntr=0.3,0.1

Type RM Length L Ch R = 1 ,39227   ,230.2,232.4,232.9
XS GIS Cut Line= 2
2266371.58929601465056.3822318272265871.42819193465001.796121484
#Sta/Elev= 30
       0  2605.7    11.5 2601.81    27.6 2593.89    43.7  2584.2    59.8 2572.63
    63.8 2571.04    71.8 2568.66    75.9 2568.33      92 2569.63      96  2569.4
     104 2567.34   108.6 2567.08     133 2567.53   140.2 2570.87   160.4 2569.66
   196.6 2568.92   204.6 2569.16   212.7    2571   236.8 2570.41   252.7 2571.52
   285.3 2571.75   307.1 2572.99   325.3 2573.47   389.7 2572.55   421.9  2573.5
   454.1 2573.17   466.2 2573.86   482.3 2573.44   494.3 2574.18   503.1 2573.89
#Mann= 4 ,-1,0
       0      .1       0      90     .05       0     104    .045       0
     133     .05       0
#XS Ineff= 2 , 0
                          332.96         2576.21
Permanent Ineff=
       F       F
Bank Sta=104,133
XS Rating Curve= 0 ,0
Exp/Cntr(USF)=0,0
Exp/Cntr=0.3,0.1

Type RM Length L Ch R = 1 ,38995   ,165.8,165.6,164.4
XS GIS Cut Line= 3
2266420.98320997464835.4581282952266141.79688671464815.302209451
2265859.23161808464924.765954258
#Sta/Elev= 30
       0 2589.86    20.9 2586.13    32.9 2582.68    40.3 2581.36    62.7 2571.38
    85.12567.003      89 2566.28      93 2566.36    97.92567.029   107.6  2568.1
   129.1  2568.3   141.2 2569.98   153.2  2569.6   169.2  2570.1   181.3 2569.03
   205.3 2569.45   225.4 2568.17   241.4 2568.02   253.8 2566.38   264.7 2565.98
   269.5 2566.42   277.5 2569.03   281.7 2569.28   298.8 2569.28   363.2 2570.54
   406.3 2570.47   458.9 2572.48   550.9 2572.69   573.3 2573.59   582.9 2574.68
#Mann= 7 ,-1,0
       0      .1       0    85.1    .045       0    97.9      .1       0
     140     .07       0   347.4     .05       0   457.4     .06       0
   537.4     .07       0
Bank Sta=85.1,97.9
XS Rating Curve= 0 ,0
Exp/Cntr(USF)=0,0
Exp/Cntr=0.3,0.1

Type RM Length L Ch R = 1 ,38829   ,266,259.2,254.5
XS GIS Cut Line= 2
2266439.61835045464673.7796163892265915.38941456 464660.35935563
#Sta/Elev= 30
       0 2588.46     3.4 2586.18    11.4 2579.41    19.4 2573.57    27.5 2569.24
    35.5 2566.65    43.5 2566.51    55.5 2567.33    79.5 2567.32    87.5 2566.87
   119.5 2567.59   127.5 2566.94   138.4 2564.47   147.5 2564.08   152.2  2564.5
   155.5 2565.15   163.5  2569.1   167.8 2570.06   171.5 2569.96   187.5 2568.28
   211.5 2568.15   327.6 2568.53   355.6 2569.12   427.6 2569.04   487.5 2570.22
   495.7 2569.41   503.6 2570.46   507.6 2571.54   519.6 2576.52   524.4 2577.09
#Mann= 6 ,-1,0
       0      .1       0      60     .07       0   138.4    .045       0
   152.2     .07       0     250     .05       0     450     .07       0
Bank Sta=138.4,152.2
XS Rating Curve= 0 ,0
Exp/Cntr(USF)=0,0
Exp/Cntr=0.3,0.1

Type RM Length L Ch R = 1 ,38570   ,210.5,207.5,205.9
XS GIS Cut Line= 3
2266533.25533349464348.1105464362266268.85001549464426.173068892
 2265938.1335225464444.639472054
#Sta/Elev= 30
       0 2582.87    30.3 2577.64    63.7 2576.19   130.5 2575.72   138.8 2575.85
   147.1 2576.72   159.2 2576.28   209.7 2576.18   214.3 2571.18     218 2566.41
   222.2 2564.45   224.62564.041   230.5 2563.66   240.82563.805   263.9 2566.31
   272.2 2568.22   275.4 2568.27   296.4 2567.49   304.4 2565.27   316.4 2564.31
   328.4 2565.87   344.5 2567.13   544.8 2568.06   568.8 2568.76   576.8 2568.41
   580.8 2568.89   592.9 2572.02   600.9 2575.59   604.9 2576.48   606.9 2576.45
#Mann= 8 ,-1,0
       0     .05       0     130      .1       0     160     .08       0
   224.6    .045       0   240.8     .08       0     260     .07       0
  355.69     .05       0  555.69     .06       0
Bank Sta=224.6,240.8
XS Rating Curve= 0 ,0
Exp/Cntr(USF)=0,0
Exp/Cntr=0.3,0.1

Type RM Length L Ch R = 1 ,38362   ,192.4,190.6,189.4
XS GIS Cut Line= 2
2266502.95997787464108.9444229222265919.95587084464358.131662216
#Sta/Elev= 30
       0 2579.66    69.3 2577.47   111.8 2575.32   137.9 2573.42   166.9 2572.18
   194.3 2571.73   224.8 2572.06   237.9 2571.74   264.4 2569.38   268.4 2568.58
   277.1 2565.43   281.4 2564.68     301 2563.44   307.1  2563.4   316.3 2563.45
   320.6 2563.94   329.3 2566.58   333.6 2567.39   346.6 2568.03   377.2 2567.56
   390.2  2566.4   398.5 2566.16   564.2 2567.64   590.3 2568.22     599 2566.96
   602.7 2567.81   608.8 2569.81   620.7 2575.45   625.1 2576.38     634 2575.98
#Mann= 6 ,-1,0
       0     .05       0     130      .1       0     301    .045       0
   316.3      .1       0     350     .07       0     450     .05       0
Bank Sta=301,316.3
XS Rating Curve= 0 ,0
Exp/Cntr(USF)=0,0
Exp/Cntr=0.3,0.1

Type RM Length L Ch R = 1 ,38172   ,62.9,59,57.2
XS GIS Cut Line= 3
2266524.98355435 463983.083961752266406.20132411463915.276515988
2265865.74799413464216.747807264
#Sta/Elev= 30
       0 2575.97    36.1 2573.76      70 2570.46   120.7  2569.1   139.1 2570.72
   152.8 2568.29   189.5 2566.53   280.3 2565.09   308.6 2565.58   329.5 2565.26
   377.8 2566.89  402.42 2564.22   410.2 2563.39  415.27 2564.21     419 2565.57
   427.8 2565.25   441.4 2566.09   450.5 2565.63     478 2566.67   487.2 2566.07
   519.3 2565.62   639.5 2566.59     707    2568   716.2 2566.76   720.8 2567.25
   724.8 2568.46   734.5 2573.63   739.1 2575.17   743.7 2575.48   755.6 2574.87
#Mann= 11 ,-1,0
       0     .05       0  166.77     .06       0  276.77     .07       0
  296.77      .1       0  386.77     .06       0  402.42    .045       0
  415.27     .06       0  496.77     .05       0  616.77     .07       0
  696.77     .05       0  726.77     .06       0
#XS Ineff= 2 , 0
          140.56 2573.37
Permanent Ineff=
       F       F
Bank Sta=402.42,415.27
XS Rating Curve= 0 ,0
Exp/Cntr(USF)=0,0
Exp/Cntr=0.5,0.3

Type RM Length L Ch R = 1 ,38113   ,55,53.5,53.4
XS GIS Cut Line= 3
2266563.74396583463723.2786245162266199.30906958463956.506609114
2265853.27079916464191.639496723
#Sta/Elev= 30
       0 2572.92       9 2572.56      28 2569.33    51.7 2570.61    77.7 2569.87
     100 2570.64     180 2568.82   209.6  2570.4   255.9 2569.06     330  2568.8
   354.3 2567.35     382 2567.21   431.6 2564.39   483.7 2563.28   497.9 2563.12
     509 2563.27     516 2563.77   528.3  2567.6   533.2 2567.85     562 2567.34
   591.2 2565.48   673.4  2566.8   683.1 2567.06   697.6 2567.83   741.1  2567.2
   772.3 2568.27     804 2567.41   813.7 2567.08     833 2575.03     851 2574.86
#Mann= 8 ,-1,0
       0     .07       0     100     .06       0     330     .07       0
   483.7    .045       0     509     .06       0   673.4     .05       0
   683.1     .07       0     804     .06       0
#XS Ineff= 3 ,-1
   14.06  214.86 2572.47  214.86     465  2568.2     545     851  2568.2
Permanent Ineff=
       F       F       F
Bank Sta=483.7,509
XS Rating Curve= 0 ,0
Exp/Cntr(USF)=0,0
Exp/Cntr=0.5,0.3

Type RM Length L Ch R = 1 ,38059   ,101.5,100.1,101.5
XS GIS Cut Line= 3
2266452.13409595463735.1692131152266162.74139536463915.537049388
 2265824.1175414 464153.57948572
#Sta/Elev= 30
       0 2570.94    42.1 2572.29   146.1 2571.07   188.5 2573.94   200.4 2574.01
   254.5 2573.87   300.5 2572.67   329.9 2572.21   334.6 2571.12   344.1 2566.76
   346.9 2566.29   383.3 2563.76   395.7 2563.62   407.7 2563.08   412.6 2563.09
   415.8  2563.7   427.3 2567.13   432.1 2567.57   451.7 2565.69   473.2 2565.72
   500.6 2565.53   524.9 2566.69   593.5 2567.15   641.1 2568.14   671.3 2568.53
     706 2570.65   719.4 2574.36     723 2574.75   740.3 2575.28   754.6 2574.41
#Mann= 9 ,-1,0
       0     .06       0   200.4      .1       0   300.5     .07       0
   395.7    .045       0   415.8     .07       0   432.1      .1       0
   473.2     .06       0   641.1     .07       0   671.3     .06       0
#XS Ineff= 2 , 0
             385  2566.5     425          2566.5
Permanent Ineff=
       F       F
Bank Sta=395.7,415.8
XS Rating Curve= 0 ,0
Exp/Cntr=0.5,0.3

Type RM Length L Ch R = 1 ,37959   ,290.4,289.9,288.6
XS GIS Cut Line= 2
2266362.98900882463659.5521095152265773.49329211464061.186553866
#Sta/Elev= 30
       0 2576.29    29.1 2575.58    95.3 2576.03   138.5 2575.43   170.2 2575.76
   226.1 2575.26   259.4 2573.48   284.1 2572.84     289 2571.73   308.3 2566.16
   322.7 2564.38   332.5 2564.31   342.2 2562.53   345.8 2562.22   365.2 2562.03
   368.8 2562.22   371.3 2562.58   380.3 2564.99   385.8 2565.25   390.6 2564.76
   400.5  2565.3   417.7 2564.87   477.7 2565.83   599.6 2566.19   656.8 2566.88
   685.9 2568.76   691.2 2569.76   700.4 2574.12   705.2 2574.67   713.3 2574.45
#Mann= 8 ,-1,0
       0     .06       0     210     .05       0     240      .1       0
   345.8    .045       0   368.8      .1       0     450     .05       0
     590     .07       0     690     .06       0
Bank Sta=345.8,368.8
XS Rating Curve= 0 ,0
Exp/Cntr(USF)=0,0
Exp/Cntr=0.3,0.1

Type RM Length L Ch R = 1 ,37669   ,333.6,332,330.7
XS GIS Cut Line= 2
2266034.40443023463527.8343948652265606.60165847463845.195501513
#Sta/Elev= 30
       0 2575.57    62.7 2575.34     120 2573.59   122.6 2573.33   125.5 2572.39
   132.3 2569.13   137.2  2566.3   142.2 2564.15   152.2 2561.88   165.5 2560.92
   177.1 2560.75   182.1 2560.98     192 2564.37   199.8 2565.49   214.1 2564.76
   230.5 2565.05   264.1 2563.83   281.7 2564.55   344.7 2565.56   361.4 2566.58
   391.3 2565.56     400 2566.12   411.2 2565.78     420 2566.51   431.9 2568.26
   462.9 2569.72   480.9 2571.22   500.8 2571.53   512.5 2573.13   532.7 2573.19
#Mann= 7 ,-1,0
       0     .05       0      60     .07       0     120      .1       0
   165.5    .045       0   182.1      .1       0     420     .05       0
     450     .06       0
#XS Ineff= 2 , 0
                           399.4         2569.32
Permanent Ineff=
       F       F
Bank Sta=165.5,182.1
XS Rating Curve= 0 ,0
Exp/Cntr(USF)=0,0
Exp/Cntr=0.3,0.1

Type RM Length L Ch R = 1 ,37337   ,158.1,158.1,161.3
XS GIS Cut Line= 2
2265936.65720939463157.1566223012265414.91555006 463607.80939374
#Sta/Elev= 30
       0 2581.52      49  2573.9    91.8 2570.31   189.7 2567.11   244.3 2567.49
   249.1  2566.3   254.3 2563.63   258.4 2562.34     306 2563.63   309.5 2562.96
   312.3 2561.38   315.2 2560.48   323.1 2560.06     335 2560.45   344.2 2560.68
   349.5 2562.61     355 2563.66   391.8 2562.72   405.9 2563.64   422.3 2563.82
   449.9 2562.66     491 2563.58     545 2563.13   571.5 2564.18   641.3 2564.48
   645.5 2565.15   649.8  2566.7     656 2569.99   661.3 2572.14   689.4 2572.04
#Mann= 10 ,-1,0
       0      .1       0      60     .05       0      70     .07       0
     220     .08       0   315.2    .045       0     335     .07       0
     380      .1       0     450     .07       0     530     .05       0
     580     .06       0
Bank Sta=315.2,335
XS Rating Curve= 0 ,0
Exp/Cntr(USF)=0,0
Exp/Cntr=0.3,0.1

Type RM Length L Ch R = 1 ,37179   ,514.2,517.2,509.7
XS GIS Cut Line= 2
2265842.44397884 463074.76811024 2265334.6178919463490.262181378
#Sta/Elev= 30
       0 2578.78     8.1  2577.8    18.4 2575.42      46 2571.77    94.3 2568.35
   176.7 2566.25   224.9 2566.33   230.3 2564.98   236.4 2562.13   247.8 2560.81
   271.7 2562.77   292.4 2562.41   301.8  2560.7   310.3 2560.17   318.8 2560.37
   328.5 2562.33   350.1 2562.25   357.5 2561.78   364.7 2560.18     375 2559.49
   385.4 2559.64  386.38  2560.2   390.6 2562.86   395.6 2563.53   490.2  2562.1
   534.9 2563.31     618 2563.41     623 2564.19   637.2 2570.91   656.1 2571.91
#Mann= 10 ,-1,0
       0     .12       0      50     .05       0     190     .07       0
     210     .08       0     320     .07       0     360      .1       0
   364.7    .045       0  386.38      .1       0     450     .07       0
     570     .06       0
Bank Sta=364.7,386.38
XS Rating Curve= 0 ,0
Exp/Cntr(USF)=0,0
Exp/Cntr=0.3,0.1

Type RM Length L Ch R = 1 ,36662   ,250,250.1,249.5
XS GIS Cut Line= 2
2265583.91433458462841.4199248332265113.86043592463285.452982676
#Sta/Elev= 30
       0 2579.59    33.6 2573.16    92.8 2568.76   225.2 2566.41   280.3 2566.58
   291.3 2564.62   302.3 2560.85   308.4 2561.46   319.4 2559.42   327.9 2560.46
   340.8 2560.25   368.3    2562   379.3 2559.13   387.3  2558.6   395.7    2559
   407.4  2561.1   424.9 2560.89   436.5 2559.59   450.8 2562.14   497.7 2561.09
   523.1  2562.9   565.6 2562.72   571.2 2563.95   582.9 2569.48   588.4 2571.17
   610.8 2570.72   627.8 2568.89   632.4 2571.67   639.1 2577.64   646.6 2582.15
#Mann= 4 ,-1,0
       0     .05       0     120     .07       0   379.3    .045       0
   395.7     .07       0
Bank Sta=379.3,395.7
XS Rating Curve= 0 ,0
Exp/Cntr(USF)=0,0
Exp/Cntr=0.3,0.1

Type RM Length L Ch R = 1 ,36412   ,199.7,195.2,194.3
XS GIS Cut Line= 2
2265452.99089006462745.0296085512265042.71914583463148.103602881
#Sta/Elev= 30
       0 2578.85    17.3 2575.67    74.4 2568.89     128 2565.68   177.1  2564.7
   188.6 2563.08   207.2 2562.11     210 2561.06   212.8 2558.83   215.7 2557.92
   229.8 2557.78   232.6 2557.87   242.3 2559.68   257.1 2559.56   266.6 2560.44
   294.9 2560.87   306.2 2560.11   317.5  2561.5   331.3 2562.01   351.4 2560.87
   379.7 2560.43   399.7 2561.59   444.8 2560.36     490    2562   518.3 2561.21
   536.7 2561.77   546.6 2563.73   557.9 2569.46   561.9 2570.79   575.1 2570.77
#Mann= 9 ,-1,0
       0     .05       0      80      .1       0     100     .07       0
   215.7    .045       0   232.6     .07       0     350     .08       0
     380      .1       0     490     .07       0     520     .06       0
Bank Sta=215.7,232.6
XS Rating Curve= 0 ,0
Exp/Cntr(USF)=0,0
Exp/Cntr=0.3,0.1

Type RM Length L Ch R = 1 ,36216   ,82.6,77.1,74.1
XS GIS Cut Line= 2
2265249.52795934462681.3319128992264960.95366383463076.378874057
#Sta/Elev= 30
       0 2584.29    24.6  2581.9    59.3 2574.11    74.1 2571.83   103.9 2569.18
   117.6 2566.06   132.5 2560.77   137.9  2559.8   148.4 2560.55   161.2 2559.79
   172.6 2561.11   183.1 2560.43     198 2561.01   215.5 2559.11   235.6 2557.98
   249.9 2557.84   253.2 2557.98   262.3 2559.96   266.8 2560.29   314.2 2558.28
   321.5 2558.63   335.8 2560.75   354.9 2560.68   375.8 2562.08   430.2 2561.06
   455.5 2562.55   460.5 2563.84   470.3 2569.11   475.4 2570.59   489.2 2570.43
#Mann= 6 ,-1,0
       0      .1       0  127.58     .07       0   235.6    .045       0
   253.2     .08       0   266.8     .07       0  447.58     .06       0
Bank Sta=235.6,253.2
XS Rating Curve= 0 ,0
Exp/Cntr(USF)=0,0
Exp/Cntr=0.5,0.3

Type RM Length L Ch R = 1 ,36139   ,44.6,47.9,51
XS GIS Cut Line= 4
2265154.42006208462596.9925045422265088.18223835 462657.92721924
2265092.28552349462764.3327030742264926.49608138463065.825754388
#Sta/Elev= 30
       0 2580.89    30.2 2577.97    68.3 2572.84   105.3 2570.41   117.3 2567.64
   125.3 2566.98   133.3 2564.43   137.3 2563.81   165.3 2563.12   185.3 2560.35
   217.8 2558.78   229.9 2560.23   235.5 2559.96   243.1  2558.4   252.2 2557.81
     262 2558.41   285.6 2558.13   296.3 2560.42   317.9 2560.91   334.4 2560.46
     368 2560.12   384.6 2561.76   412.2 2561.93   437.5 2561.18   466.8  2561.1
   491.7 2563.25   500.6  2565.4   507.9 2568.89   512.4 2570.16   540.6 2569.65
#Mann= 7 ,-1,0
       0      .1       0   217.8     .08       0   243.1    .045       0
     262     .08       0   317.9    .045       0   334.4     .08       0
   437.5     .07       0
#XS Ineff= 2 , 0
           223.9  2561.6   281.2            2561
Permanent Ineff=
       F       F
Bank Sta=243.1,262
XS Rating Curve= 0 ,0
Exp/Cntr(USF)=0,0
Exp/Cntr=0.5,0.3

Type RM Length L Ch R = 1 ,36091   ,91.3,94.3,102.9
XS GIS Cut Line= 4
2265129.98125522462591.7159319352265034.77247816462673.997574171
2265046.29696464462758.1415722272264876.34904634463027.091676366
#Sta/Elev= 30
       0 2578.27    39.4 2573.71    61.9 2571.92    65.8  2571.2    76.4 2567.11
   113.4 2564.25   118.7 2563.02   124.6  2559.7     129 2558.94   161.3 2559.88
   177.5 2559.41   210.8 2560.16   217.4 2559.15   237.72558.407   256.9 2558.16
   261.62558.415   266.7  2558.9   280.6 2558.61     357 2560.41     372 2561.39
   382.7 2561.24   409.4 2562.95   422.6 2561.85   446.9 2563.34   476.8 2562.24
   484.2 2562.89   493.5 2567.46   499.3 2569.48   507.7 2569.96   528.9 2569.42
#Mann= 8 ,-1,0
       0      .1       0  165.84     .08       0   237.7    .045       0
   261.6     .08       0  280.77     .05       0  390.77     .07       0
  470.77     .06       0  510.77     .07       0
#XS Ineff= 2 , 0
           232.7    2561   266.6          2560.6
Permanent Ineff=
       F       F
Bank Sta=237.7,261.6
XS Rating Curve= 0 ,0
Exp/Cntr(USF)=0,0
Exp/Cntr=0.5,0.3

Type RM Length L Ch R = 1 ,35997   ,208.8,204.7,201.6
XS GIS Cut Line= 3
2265123.11172877462577.5493494432265005.96330248462682.961315329
2264751.18580606462918.316312019
#Sta/Elev= 30
       0 2579.52    44.3 2573.45    63.1 2572.05    68.5 2570.67    73.9 2567.99
    77.2 2567.25    95.3 2566.53   111.6 2564.58   127.7 2559.29   137.8 2558.68
   143.9 2556.79   149.2  2556.6   160.9 2558.35   170.9 2556.83   178.52557.523
   187.3 2556.35   194.4 2556.46   200.1  2557.6   205.7 2559.09   214.5 2558.39
   225.5 2560.15   262.3 2559.44   273.7 2560.17   312.5 2559.54   328.8 2559.47
   372.4 2561.71     452 2564.41     465 2565.53   477.5 2568.93   504.4  2569.2
#Mann= 7 ,-1,0
       0      .1       0   111.6     .08       0   178.5    .045       0
   200.1     .07       0   312.5     .05       0   372.4     .07       0
     452     .06       0
Bank Sta=178.5,200.1
XS Rating Curve= 0 ,0
Exp/Cntr(USF)=0,0
Exp/Cntr=0.3,0.1

Type RM Length L Ch R = 1 ,35792   ,324.9,325.2,330
XS GIS Cut Line= 4
2264924.63837845  462492.97647242264866.44572942462550.595506304
2264860.01188884462566.0802402732264622.74608217462828.156482043
#Sta/Elev= 30
       0 2571.72      23 2566.11    28.8 2565.25    57.1 2561.99    68.4 2561.71
      74 2559.85    79.9 2556.81    82.5 2556.06    84.7 2555.55    87.8 2555.48
    98.7 2555.98   104.4 2557.76   113.6 2558.25   123.4 2558.15   143.2 2556.82
   151.4 2557.43   167.6 2557.02   189.2  2559.1   205.5 2558.41     214 2558.47
     248 2559.98   348.7 2561.35   360.7 2562.42   375.4 2564.75   399.6 2566.68
   412.2 2568.17     432    2569   446.2 2569.03   449.1  2569.4   452.2 2570.37
#Mann= 7 ,-1,0
       0      .1       0   67.18     .08       0    82.5    .045       0
    98.7     .08       0  177.18     .07       0  287.18     .05       0
  397.18     .06       0
Bank Sta=82.5,98.7
XS Rating Curve= 0 ,0
Exp/Cntr(USF)=0,0
Exp/Cntr=0.3,0.1

Type RM Length L Ch R = 1 ,35467   ,317.1,312.2,314.9
XS GIS Cut Line= 3
2264750.99792668462359.7160332762264686.53835969462379.196519971
2264442.78935763462628.305398496
#Sta/Elev= 30
       0 2594.68    11.3 2593.98    22.7 2592.35    44.7  2583.4      58 2578.53
    81.3 2571.02    93.6  2568.2     110 2561.55   121.3 2557.87   126.1  2556.7
   132.6 2556.47   139.4 2555.11   145.1 2554.59   150.8 2555.14   156.5 2557.39
   175.1 2557.62   185.1 2557.06   196.5 2555.22   225.1  2555.6   228.8 2555.08
   234.5 2554.59   243.6 2555.06   259.9 2558.29   271.2 2558.22   288.4 2559.97
   299.6 2559.03   322.2 2560.13   330.6 2561.26   361.8 2562.99   415.9 2568.64
#Mann= 6 ,-1,0
       0      .1       0  117.34     .08       0   228.8    .045       0
   243.6     .08       0  317.34     .07       0  397.34     .06       0
#XS Ineff= 2 , 0
                          289.16         2571.62
Permanent Ineff=
       F       F
Bank Sta=228.8,243.6
XS Rating Curve= 0 ,0
Exp/Cntr(USF)=0,0
Exp/Cntr=0.3,0.1

Type RM Length L Ch R = 1 ,35155   ,156,149.1,142.9
XS GIS Cut Line= 3
2264587.64707164 462153.063018352264418.38781476462333.292782619
2264452.86655227462607.555467375
#Sta/Elev= 30
       0 2582.65    16.7 2580.51    39.3 2574.03    50.6 2571.54    60.5 2569.85
    71.5  2569.1      77 2566.08    81.8 2561.56    87.4  2555.1    93.4 2552.93
   104.4 2552.56   110.82552.731   124.2 2553.12   132.7 2554.55   145.3 2554.83
   155.3 2555.92   181.2 2555.62   203.2 2557.14   228.9 2557.26   323.7 2560.64
     364 2560.77   412.4 2562.22   417.1 2561.89   424.5 2559.31   428.5 2559.27
   436.6 2561.87   440.6  2562.6     454  2563.3   494.1 2563.95   523.7 2566.58
#Mann= 5 ,-1,0
       0      .1       0    93.4    .045       0   110.8     .07       0
  247.25     .06       0  257.25     .07       0
#XS Ineff= 2 , 0
                          322.29         2569.69
Permanent Ineff=
       F       F
Bank Sta=93.4,110.8
XS Rating Curve= 0 ,0
Exp/Cntr(USF)=0,0
Exp/Cntr=0.3,0.1

Type RM Length L Ch R = 1 ,35006   ,167.5,148.4,129
XS GIS Cut Line= 4
2264517.86645008461999.948139256 2264425.9104484462090.562470533
2264345.81647738462270.5430456552264436.71496718462599.658267363
#Sta/Elev= 30
       0 2604.82    13.6 2603.79    24.5 2602.22    44.5  2597.6    75.4 2591.86
    98.6 2586.28   115.7 2579.84   123.7 2576.23   127.1 2574.01     132  2569.6
   145.1 2556.75   149.5 2554.07   155.72552.069   171.4 2551.36   174.8 2551.98
   188.9  2555.1   231.8 2557.24   298.3 2556.49   320.2 2557.69   346.4 2557.82
   378.9 2559.15   449.2 2560.03   507.3 2561.94   552.9 2562.26   573.7 2562.93
   586.1 2561.92   594.4 2561.49   598.6 2564.01   609.8 2564.86   667.5 2567.32
#Mann= 8 ,-1,0
       0      .1       0      10     .12       0   155.7    .045       0
   174.8     .07       0   376.1     .06       0   476.1     .07       0
   586.1     .06       0   606.1     .07       0
Bank Sta=155.7,174.8
XS Rating Curve= 0 ,0
Exp/Cntr(USF)=0,0
Exp/Cntr=0.5,0.3

Type RM Length L Ch R = 1 ,34858   ,103.5,110.4,124.6
XS GIS Cut Line= 5
2264436.61883222461508.2845861642264300.99201657461825.959135878
2264287.02812788461926.2452455792264298.40611126462196.966023663
2264417.81224812 462595.93203314
#Sta/Elev= 30
       0 2581.26    35.8 2583.31    61.9 2583.83   148.8 2582.56     193 2583.33
   215.1 2582.92   296.6 2576.91   345.4 2571.47   368.9 2572.73     385 2572.64
   397.1 2570.68   413.3 2564.44   425.4 2562.22   477.8 2559.14   485.6 2557.54
   493.6 2554.07   497.6 2553.28   525.7 2553.44   537.7 2551.83   546.6 2551.13
   565.7 2551.09   582.3 2551.83   589.7 2553.68   597.7 2552.95   613.8 2554.58
   645.8 2554.85   713.8  2557.2   930.8 2560.34  1031.1 2565.27  1134.1 2568.33
#Mann= 11 ,-1,0
       0     .06       0     240     .08       0     300     .06       0
  445.42     .07       0   537.7    .045       0   582.3     .07       0
  646.67     .06       0  797.63     .07       0  847.63     .06       0
  947.63     .07       0 1057.63     .06       0
#XS Ineff= 2 , 0
             420  2568.1     640         2567.59
Permanent Ineff=
       F       F
Bank Sta=537.7,582.3
XS Rating Curve= 0 ,0
Exp/Cntr(USF)=0,0
Exp/Cntr=0.5,0.3

Type RM Length L Ch R = 1 ,34747   ,150.1,184.3,207.6
XS GIS Cut Line= 4
2264350.01451245461472.7087979132264207.82106452461813.013937158
2264204.01273124462178.6139320152264324.60995177462614.033370334
#Sta/Elev= 30
       0 2566.16   127.1 2566.57   147.9  2568.2   225.9 2570.93   299.6  2570.1
   308.3 2568.99   334.3 2561.16   344.2 2557.22     377 2553.44     401 2555.02
     433 2553.96     481  2556.3     497 2555.07     509  2552.1     529 2551.42
   533.82552.006   542.8 2553.64     577 2552.94     581 2553.49     593 2558.33
     597 2559.14     609 2558.43     621 2556.11     693 2554.26     733 2556.64
   757.9 2555.71     795 2556.03   882.9 2559.81  1077.4 2564.33  1186.2 2568.36
#Mann= 13 ,-1,0
       0     .06       0      80      .1       0     280     .06       0
     340     .08       0  388.82     .07       0     509    .045       0
   533.8     .07       0  578.82     .06       0  784.44     .07       0
  804.44     .06       0  984.44     .07       0 1084.44      .1       0
 1174.44     .06       0
#XS Ineff= 2 , 0
          468.44 2567.99     600         2567.62
Permanent Ineff=
       F       F
Bank Sta=509,533.8
XS Rating Curve= 0 ,0
Exp/Cntr(USF)=0,0
Exp/Cntr=0.5,0.3

Type RM Length L Ch R = 1 ,34563   ,197.4,182.4,162.5
XS GIS Cut Line= 4
2264318.41923141461460.4475008192264150.42169796461819.041728574
2264036.19663613461847.0242772852263826.08262848462176.316641792
#Sta/Elev= 30
       0 2558.29    24.1 2557.03    71.5 2557.55   137.3 2556.19   184.4 2554.08
   197.8 2558.56     204 2559.64   212.8 2564.52   217.3 2565.93   230.5 2567.95
   248.9 2568.35   270.3 2566.73     297 2556.74     306 2554.94   344.7 2553.58
   363.2 2551.97   402.4 2554.25   414.8 2551.03     423 2552.03  433.722551.617
   443.6 2550.78455.07482551.539   464.2 2553.32   509.5 2555.32   555.7 2554.57
   744.2 2556.07   838.8 2558.53   862.8 2565.33   885.9 2573.84   904.2 2578.05
#Mann= 8 ,-1,0
       0      .1       0     230     .08       0     426     .07       0
  433.72    .045       0455.0748     .07       0   603.6      .1       0
   723.6     .07       0   903.6     .05       0
#XS Ineff= 2 , 0
          246.99 2574.75  699.72         2559.42
Permanent Ineff=
       F       F
Bank Sta=433.72,455.0748
XS Rating Curve= 0 ,0
Exp/Cntr(USF)=0,0
Exp/Cntr=0.3,0.1

Type RM Length L Ch R = 1 ,34381   ,183.6,181.2,179
XS GIS Cut Line= 3
2264043.05971567461514.7885298312264039.17302162461620.810647681
2263767.32384849462131.644488231
#Sta/Elev= 30
       0 2591.96    18.4 2582.86    30.4 2575.65    34.4 2572.64    38.4  2568.4
    50.4 2554.43    54.4 2552.82    70.4 2551.91   108.6 2552.88   120.4 2551.94
   133.7 2554.69   165.4  2554.5   169.9 2554.34   183.5 2551.01   191.4 2550.21
   203.2 2549.94   212.1 2550.34   253.5 2552.46   265.3 2554.16   291.3 2553.19
   374.7 2554.55   414.6 2553.86   478.2  2555.5   599.5 2556.12   614.3  2557.5
   627.6 2560.95   655.7 2573.26   661.6 2575.16   668.4 2576.35   684.8  2577.5
#Mann= 9 ,-1,0
       0      .1       0  116.09     .08       0  146.09     .07       0
   191.4    .045       0   212.1     .07       0  226.09      .1       0
  346.09     .07       0  456.09      .1       0  676.09     .05       0
#XS Ineff= 2 , 0
          102.93 2562.76  477.97         2561.78
Permanent Ineff=
       F       F
Bank Sta=191.4,212.1
XS Rating Curve= 0 ,0
Exp/Cntr(USF)=0,0
Exp/Cntr=0.3,0.1

Type RM Length L Ch R = 1 ,34199   ,281,287.8,292.4
XS GIS Cut Line= 3
2263867.60995819461548.9694964282263764.78495964461802.858381745
2263630.22385042462021.202823118
#Sta/Elev= 30
       0 2574.87      12 2566.83    17.5 2563.56    34.8 2554.34    39.1 2552.88
    47.7 2552.38      52 2551.41    56.3 2549.49    59.4  2548.9    76.5  2548.5
    83.7 2548.78    90.9 2551.08   108.1 2552.84   125.4 2552.54   162.5 2553.16
   207.4 2553.06   245.5 2552.25   284.8 2553.12   304.8 2552.96   334.2 2554.11
   375.3 2553.83   412.3    2555   455.2 2554.92   464.6 2556.14   482.5 2559.97
   497.5 2563.98   506.9 2567.36   520.2 2571.18   525.7 2572.07   530.4 2572.38
#Mann= 5 ,-1,0
       0     .08       0    59.4    .045       0    83.7     .08       0
      90     .07       0  423.92      .1       0
Bank Sta=59.4,83.7
XS Rating Curve= 0 ,0
Exp/Cntr(USF)=0,0
Exp/Cntr=0.3,0.1

Type RM Length L Ch R = 1 ,33912   ,166.6,181.5,188.4
XS GIS Cut Line= 2
2263669.57662765 461474.072275262263376.33496511461891.719491606
#Sta/Elev= 30
       0 2566.34    28.2 2555.46    43.4 2552.04    57.6 2551.41      86 2551.95
   101.5 2551.02   118.1 2550.94   138.3 2552.34   152.5 2550.75   165.1 2551.66
     170 2551.25   178.4 2547.82   181.3  2547.3   190.4  2547.1   207.1 2547.28
   211.3 2547.79   218.6 2549.66   235.8 2549.91   243.3  2551.5   278.9  2551.5
   322.6 2553.31   365.5 2554.16   419.2 2554.13   468.1 2556.49   482.8 2560.03
   487.7 2562.44   494.2 2567.39   497.1 2569.05   502.9 2570.01   510.3 2570.09
#Mann= 5 ,-1,0
       0      .1       0   181.3    .045       0   207.1     .07       0
     310      .1       0     410     .06       0
Bank Sta=181.3,207.1
XS Rating Curve= 0 ,0
Exp/Cntr(USF)=0,0
Exp/Cntr=0.3,0.1

Type RM Length L Ch R = 1 ,33730   ,325.5,311,299.2
XS GIS Cut Line= 4
2263605.62961446461349.1762295162263462.84484592461503.815041102
2263362.69830448461554.1999248792263197.02922884461745.657057177
#Sta/Elev= 30
       0 2557.41    72.9 2555.04   125.2 2551.24   226.9 2551.38   231.4 2550.84
   240.4 2547.46   244.8 2547.19   264.1 2547.39   270.1 2548.09     276 2550.95
   280.6 2551.96   299.9 2550.85   320.7 2551.18     352 2547.85   371.9  2547.5
   397.4 2547.73   405.9 2549.85   416.4 2550.77   442.9 2549.56   471.1 2551.05
   485.2 2552.72   522.2 2552.47   528.2 2553.26   534.3 2556.84   540.4 2558.98
   556.2 2560.56     559 2561.81   564.8 2566.49   567.5 2567.33   575.8 2567.89
#Mann= 9 ,-1,0
       0      .1       0      10     .07       0      80      .1       0
     120     .07       0   240.4    .045       0   264.1     .07       0
  414.96     .06       0  514.96      .1       0  544.96     .06       0
#XS Ineff= 2 , 0
                          485.75         2555.46
Permanent Ineff=
       F       F
Bank Sta=240.4,264.1
XS Rating Curve= 0 ,0
Exp/Cntr(USF)=0,0
Exp/Cntr=0.3,0.1

Type RM Length L Ch R = 1 ,33419   ,346.1,343.9,341.1
XS GIS Cut Line= 3
2263319.20996591461165.5972795992263258.27663343461212.566723383
2263037.39330321461636.561161863
#Sta/Elev= 30
       0  2576.3    30.4 2572.15    69.5  2565.1    82.1 2559.93    95.7 2551.81
   104.7 2549.18   113.7 2548.38   124.8 2548.38   149.8 2549.41   154.3 2548.71
     162 2546.24   170.9  2545.8   182.7 2546.34   194.9 2548.94   226.5 2549.24
     240 2548.54   280.6 2550.12   316.7 2548.18   339.2 2549.09   349.9 2550.21
   374.7  2550.9     479 2550.78   506.1 2551.66   515.1 2552.95   519.6 2554.41
   523.8 2556.53   533.2  2564.1   537.7 2565.61   550.4 2566.39     555 2570.22
#Mann= 6 ,-1,0
       0      .1       0     162    .045       0   182.7      .1       0
  326.94     .05       0  336.94      .1       0  546.94     .06       0
Bank Sta=162,182.7
XS Rating Curve= 0 ,0
Exp/Cntr(USF)=0,0
Exp/Cntr=0.3,0.1

Type RM Length L Ch R = 1 ,33075   ,251.5,238.8,224.1
XS GIS Cut Line= 2
2262935.83774908461062.7722810462262772.07941805461498.191719365
#Sta/Elev= 30
       0 2569.01     6.8  2565.9    23.9 2556.57    36.8 2552.44      41 2551.69
    51.3 2550.89    62.4 2548.57    96.6 2547.02   105.1 2547.49   109.4 2547.16
   116.5 2545.56   130.8 2545.42   135.1 2545.59   143.6 2548.36   147.6 2548.73
     165 2548.44   169.3    2548   190.6 2548.14   207.7 2547.23   318.4 2548.03
   378.6 2547.76     400 2548.58   421.4 2549.45   430.2 2550.35   438.5 2551.78
   442.6 2553.36   451.3 2559.48   455.6 2561.53   459.8 2562.22   465.2 2562.38
#Mann= 4 ,-1,0
       0      .1       0   116.5    .045       0   135.1      .1       0
     400     .06       0
Bank Sta=116.5,135.1
XS Rating Curve= 0 ,0
Exp/Cntr(USF)=0,0
Exp/Cntr=0.3,0.1

Type RM Length L Ch R = 1 ,32836   ,211.2,227,239.4
XS GIS Cut Line= 4
2262664.17664179460990.4139487312262634.97941998461083.083391871
2262677.01266115461206.4188889662262602.85063564 461488.50402491
#Sta/Elev= 30
       0 2565.45     8.6 2563.08    40.5 2556.38    56.4 2551.76      70 2546.89
    82.6 2546.01   103.6 2547.46   150.2 2548.18   169.1 2547.31   178.5 2546.16
183.06292544.946   188.1 2544.18203.95382545.224   213.2 2547.26   221.9 2546.77
   234.5 2548.01   246.8 2547.97   259.3 2546.72   286.3 2546.37   317.2 2547.53
   416.4 2547.03   466.1 2548.31   470.2 2549.75   472.8 2551.37   486.7 2562.32
   490.9 2563.31   499.2 2563.47   503.3 2564.54   511.6 2570.75   519.1 2578.59
#Mann= 7 ,-1,0
       0     .12       0      50      .1       0  157.16     .08       0
183.0629    .045       0203.9538     .08       0  257.46      .1       0
  467.46     .06       0
Bank Sta=183.0629,203.9538
XS Rating Curve= 0 ,0
Exp/Cntr(USF)=0,0
Exp/Cntr=0.3,0.1
