HEC-RAS study THRNYCK.prj: THRNYCK

--- THRNYCK.g01 (geometry) --- (continued)

Type RM Length L Ch R = 1 ,32609   ,376.9,363.6,353.9
XS GIS Cut Line= 2
2262542.30997684460951.0611715062262351.89331285461381.402832119
#Sta/Elev= 30
       0 2564.43    28.6 2558.76    32.9 2557.32    50.4 2549.53    59.2 2546.41
    63.9 2545.26    67.9 2545.06    85.1 2546.65    94.2 2546.62     151 2544.46
   163.9 2544.81     186 2546.33   203.5 2546.56   216.6 2545.53   225.4 2543.55
   232.6  2543.1   239.7 2543.41   247.3 2544.23   251.6 2546.43   260.4 2547.21
   303.4 2546.54     326    2547   433.8 2547.04   435.3 2547.25   439.7 2550.13
   444.1 2554.78   448.5 2557.56   452.8 2558.23     466  2558.7   470.6 2562.49
#Mann= 5 ,-1,0
       0     .12       0     100      .1       0   225.4    .045       0
   239.7      .1       0     420     .06       0
Bank Sta=225.4,239.7
XS Rating Curve= 0 ,0
Exp/Cntr(USF)=0,0
Exp/Cntr=0.3,0.1

Type RM Length L Ch R = 1 ,32246   ,258.1,265.1,270.4
XS GIS Cut Line= 3
2262238.91275889460924.402838548 2262274.1977356461041.772171324
2262223.61722738461351.204442778
#Sta/Elev= 30
       0 2577.09     9.2 2573.41    21.7 2567.18    42.6 2558.05    67.6 2543.96
    69.1 2543.36    71.8 2542.43      76 2542.16    80.2 2542.24    84.3 2542.82
    92.7 2543.93     126 2546.85   174.6 2545.78   203.9 2545.91   227.3 2545.61
   256.2 2545.79     276 2546.27   303.5 2546.33   308.4 2546.06   346.8  2546.4
     392 2547.28   393.5 2547.44   397.6 2549.83   401.6 2553.72   405.7 2556.52
   409.7 2557.35   421.9 2557.74   425.9  2560.1   432.6 2566.35   436.1 2569.04
#Mann= 7 ,-1,0
       0      .1       0      50     .12       0    69.1    .045       0
    84.3     .12       0     120      .1       0  322.56     .06       0
  422.56      .1       0
Bank Sta=69.1,84.3
XS Rating Curve= 0 ,0
Exp/Cntr(USF)=0,0
Exp/Cntr=0.3,0.1

Type RM Length L Ch R = 1 ,31980   ,279.3,287.1,291.1
XS GIS Cut Line= 3
2262067.96478139460861.7632998832262005.99962321461001.387127374
2261998.99425671461289.101457906
#Sta/Elev= 30
       0 2571.41    11.5 2569.53    19.2 2568.86    38.9 2565.34    56.3 2560.51
    75.2 2554.63    86.9 2550.52    95.6 2546.76     100 2545.59   104.4 2545.15
   125.2 2544.79   148.2 2542.19   164.6 2544.43   180.6 2544.66   200.6 2541.75
   212.6  2541.4   220.6  2541.6   228.6 2543.13   252.6 2543.07   261.4 2544.11
   271.5  2544.7   300.6 2544.65   347.5 2547.38   368.6 2546.72   380.6  2546.8
   384.8 2547.53   396.6 2550.61   416.6 2557.56   424.6 2560.87   440.6 2561.09
#Mann= 6 ,-1,0
       0     .12       0  192.76      .1       0   200.6    .045       0
   220.6      .1       0  292.76     .06       0  392.76      .1       0
Bank Sta=200.6,220.6
XS Rating Curve= 0 ,0
Exp/Cntr(USF)=0,0
Exp/Cntr=0.3,0.1

Type RM Length L Ch R = 1 ,31693   ,304.2,291.4,278.2
XS GIS Cut Line= 3
2261771.08976488460897.4418822762261697.05957279461114.722957726
2261734.50980699461340.144264644
#Sta/Elev= 30
       0 2559.66    25.1 2553.63    50.4  2548.6      59 2546.31      80 2541.73
100.40042540.986   113.8 2540.12  119.78 2540.92   130.7 2542.06   155.1 2542.94
   168.8 2542.68   185.7 2543.41   202.6 2543.21   223.7 2545.12   260.4 2544.11
   268.5 2544.35   276.6 2543.89   324.8 2543.85   353.7 2544.78   382.1 2544.58
   386.1 2545.38   390.2 2546.79   414.5 2556.74   418.6 2559.03   429.1 2565.96
   434.8 2570.29   438.8 2572.52   442.9 2573.29   455.1 2574.31   458.1 2576.37
#Mann= 5 ,-1,0
       0     .12       0100.4004    .045       0  119.78     .12       0
  359.55      .1       0  458.06     .06       0
Bank Sta=100.4004,119.78
XS Rating Curve= 0 ,0
Exp/Cntr(USF)=0,0
Exp/Cntr=0.3,0.1

Type RM Length L Ch R = 1 ,31402   ,388,381.7,371.8
XS GIS Cut Line= 2
2261421.39054816460836.8111731142261641.00443396461353.475054734
#Sta/Elev= 30
       0 2576.36    52.6 2568.65    66.5 2564.99    69.5 2563.75    74.3 2560.68
    87.8 2549.19    91.7 2546.51   112.2 2541.49   117.8 2540.18   121.4  2539.9
   127.5 2541.09   139.7 2542.22   152.5 2541.46     209 2542.82   235.1 2542.46
   265.5 2543.07   283.2 2542.53     344 2543.13   365.5 2542.53   387.2 2543.48
   426.3 2544.16   465.5 2543.84   487.2 2544.84   493.4 2546.27   504.6 2550.75
   513.3 2552.38     522 2557.52   549.1 2571.81   556.7  2576.8   561.4 2578.93
#Mann= 5 ,-1,0
       0      .1       0   112.2    .045       0   127.5     .12       0
     330      .1       0     540     .06       0
Bank Sta=112.2,127.5
XS Rating Curve= 0 ,0
Exp/Cntr(USF)=0,0
Exp/Cntr=0.3,0.1

Type RM Length L Ch R = 1 ,31020   ,227,229,234.4
XS GIS Cut Line= 6
2261144.71386156461069.8594003972261232.31664615461122.757374449
2261297.86483796461270.6703339262261308.96721007 461286.18926192
2261338.21519125461301.2342768282261411.16680085461450.786691685
#Sta/Elev= 30
       0 2575.32    18.1 2571.04      37 2565.05      69 2558.11    76.1 2555.59
    83.6 2551.29    92.8 2548.33   104.1 2542.95   109.4 2541.78   131.3 2541.31
   153.1 2541.96   201.2 2542.09   231.9 2541.36     260 2542.11   267.2 2541.24
   284.92537.646   304.8 2537.45   309.3 2537.61   316.1 2539.32   338.5 2540.04
   353.4 2541.71   402.7 2541.74   409.5 2542.47   419.2 2544.47   422.8 2545.45
     430 2549.94   442.1 2556.21   467.3 2571.01   476.3 2575.58   482.5 2580.04
#Mann= 6 ,-1,0
       0      .1       0  122.33     .12       0  232.33      .1       0
282.5599    .045       0   284.9    .045       0   309.3      .1       0
Bank Sta=284.9,309.3
XS Rating Curve= 0 ,0
Exp/Cntr(USF)=0,0
Exp/Cntr=0.3,0.1

Type RM Length L Ch R = 1 ,30791   ,555.4,549,532.2
XS GIS Cut Line= 2
2260956.77388803461185.9083904252261274.13499468 461562.93338512
#Sta/Elev= 30
       0 2578.63     5.3 2577.42      20 2572.15    38.8 2562.69    46.1 2557.06
    61.8 2542.52      67 2539.65    79.8 2538.04    93.2 2538.04   108.8 2539.27
   129.8 2538.91   160.9 2540.13   217.6 2541.05   234.3  2539.4   244.8 2539.53
   265.7 2538.37   284.8 2539.74   302.3 2539.76     318 2538.94   328.4  2540.1
   365.3 2540.77   390.8 2539.14   399.3 2537.26   402.8 2536.84   415.2 2537.26
   440.1 2551.58   461.8 2567.24     476 2574.64   489.8 2583.81   492.8 2584.83
#Mann= 8 ,-1,0
       0      .1       0      70     .12       0     180      .1       0
     200     .12       0     320      .1       0   399.3    .045       0
   415.2      .1       0     490     .06       0
Bank Sta=399.3,415.2
XS Rating Curve= 0 ,0
Exp/Cntr(USF)=0,0
Exp/Cntr=0.3,0.1

Type RM Length L Ch R = 1 ,30242   ,239.8,232.4,221.7
XS GIS Cut Line= 2
2260776.75130493461400.9621247322261085.56705126461722.715174271
#Sta/Elev= 30
       0  2556.4    10.7 2555.02    28.1 2550.93    44.7 2545.27      62  2537.4
    66.8 2536.14    73.3 2535.88   100.1 2536.02   107.2 2538.23   111.2 2538.99
   126.3  2539.5   149.4 2538.52   155.3 2537.72   163.8 2537.71   172.5 2538.84
   183.6 2541.02   188.8 2541.45   207.1 2540.57   279.8 2539.61   293.8 2539.26
   299.7 2538.73   305.3 2539.35   327.4 2540.06   363.1 2542.83   393.9 2545.89
   403.5 2546.36   415.6 2548.29   426.6 2551.95   432.8 2555.21     446 2563.26
#Mann= 7 ,-1,0
       0     .12       0      50      .1       0    66.8    .045       0
   100.1      .1       0     290     .12       0     320      .1       0
     430     .06       0
Bank Sta=66.8,100.1
XS Rating Curve= 0 ,0
Exp/Cntr(USF)=0,0
Exp/Cntr=0.3,0.1

Type RM Length L Ch R = 1 ,30010   ,361.1,373.5,377.3
XS GIS Cut Line= 4
2260548.14343669461503.1388430522260685.15918849461638.383736121
2260762.31987485461676.964079301 2260961.3021312461856.672058044
#Sta/Elev= 30
       0  2576.7    35.4 2561.38    48.5 2557.07    54.2  2553.3    67.5 2541.95
    71.2 2539.66      75 2538.45   101.2 2536.74   133.9 2538.44   168.3 2538.65
   191.1 2538.15   200.4 2536.86   213.8 2537.13220.78332536.144   227.2  2535.6
243.5758 2535.93   253.5 2537.94   278.8 2535.97   297.2 2538.13   356.7 2539.03
   396.4 2539.28   426.8 2537.59   446.2 2537.31   461.5 2538.17   475.7 2538.16
   480.7  2539.3   486.1 2541.85   523.8 2565.72   529.5 2568.25   546.9 2572.95
#Mann= 5 ,-1,0
       0      .1       0     180     .12       0     190      .1       0
220.7833    .045       0243.5758      .1       0
#XS Ineff= 2 , 0
          136.75 2549.62
Permanent Ineff=
       F       F
Bank Sta=220.7833,243.5758
XS Rating Curve= 0 ,0
Exp/Cntr(USF)=0,0
Exp/Cntr=0.3,0.1

Type RM Length L Ch R = 1 ,29637   ,213.1,214.9,216.4
XS GIS Cut Line= 2
 2260410.8486795461629.6941467792260716.08798872462112.215504136
#Sta/Elev= 30
       0 2568.19      42 2551.22    56.2 2543.16    62.3 2540.57    69.8 2537.71
    79.9 2536.46   136.8 2537.16   165.1  2535.8   193.4 2537.19   219.5 2536.62
   267.3 2537.36   293.4 2535.94   309.2 2536.27   322.4 2534.39   346.7 2536.56
   387.5 2536.47411.2668 2534.84   425.4 2533.89426.05532533.909   429.7 2534.16
   436.4  2536.4   457.8 2537.99   481.8 2538.12   493.4 2537.29     520 2537.87
   529.5 2538.98   533.7  2540.8     539 2544.43   548.5 2554.43     571  2571.5
#Mann= 5 ,-1,0
       0      .1       0     240     .12       0     320      .1       0
411.2668    .045       0426.0553      .1       0
#XS Ineff= 2 , 0
          183.13 2549.62
Permanent Ineff=
       F       F
Bank Sta=411.2668,426.0553
XS Rating Curve= 0 ,0
Exp/Cntr(USF)=0,0
Exp/Cntr=0.3,0.1

Type RM Length L Ch R = 1 ,29422   ,262.6,276.4,284.5
XS GIS Cut Line= 2
2260297.93223064461787.6250486262260522.62389414462234.469486784
#Sta/Elev= 30
       0 2563.73    14.7 2558.14    38.6 2546.94    44.5  2544.9    89.2 2538.96
   101.1  2537.9   113.7 2535.89   122.6 2535.44   136.1 2535.77   156.4 2534.37
   171.9 2534.91   185.3 2534.05   202.4 2534.67   221.1 2536.15   230.1 2536.25
   252.5 2534.73   300.7 2534.93   312.7 2534.03   321.6 2532.76   328.6 2532.08
   337.5 2532.26   342.5 2532.89   364.4 2538.09   368.9 2538.47   387.1 2541.77
   400.2 2543.25   414.6 2545.55   449.5 2555.93   462.9 2560.38   500.2 2567.67
#Mann= 5 ,-1,0
       0      .1       0      50     .12       0     190      .1       0
   321.6    .045       0   342.5      .1       0
Bank Sta=321.6,342.5
XS Rating Curve= 0 ,0
Exp/Cntr(USF)=0,0
Exp/Cntr=0.3,0.1

Type RM Length L Ch R = 1 ,29145   ,310.7,294,279
XS GIS Cut Line= 4
2260149.25434426461849.0302722392260224.91591452461971.714468941
2260214.48122012462096.5319785022260322.82268332462276.208264394
#Sta/Elev= 30
       0 2572.39      11 2569.89    19.7 2565.81    23.7 2562.67    37.1 2549.62
    51.3 2536.79    56.6 2534.68    61.3 2534.27    74.9 2535.59    83.6 2535.01
    89.6 2535.44    94.2 2535.31    98.9 2533.92     104 2533.27   141.2 2533.26
180.50552532.408 203.0022532.212   209.8 2532.16   246.2    2535   284.2  2535.7
     341 2535.34   363.6 2536.26   378.9  2537.5     408 2541.75   419.9  2542.8
   425.5 2543.82   434.3 2546.99     457 2559.38     471  2566.4   479.2 2569.83
#Mann= 5 ,-1,0
       0     .12       0      80      .1       0      90     .12       0
180.5055    .045       0 203.002      .1       0
Bank Sta=180.5055,203.002
XS Rating Curve= 0 ,0
Exp/Cntr(USF)=0,0
Exp/Cntr=0.3,0.1

Type RM Length L Ch R = 1 ,28851   ,330.4,325.8,321.6
XS GIS Cut Line= 2
2259859.97390346461955.1917129362260198.91556536462372.838929282
#Sta/Elev= 30
       0 2573.94      18 2563.02    24.3 2560.19    33.5 2554.17    41.4 2550.26
    64.1 2535.42    70.1 2532.28    76.5 2531.19    92.6 2532.62     1102531.662
   126.2 2530.57   131.3 2531.72     140 2533.15     159 2532.14   192.1 2534.15
     255 2533.87   270.4 2533.27   301.3 2534.92     340 2535.32   359.9 2534.83
   405.4  2535.2   422.4  2535.7     431 2536.92   438.3 2539.01   444.7 2541.89
   476.4 2559.81   489.1 2564.69   497.1 2566.82   527.2 2569.58   537.9 2571.09
#Mann= 5 ,-1,0
       0      .1       0     110    .045       0   131.3      .1       0
     220     .12       0     340      .1       0
Bank Sta=110,131.3
XS Rating Curve= 0 ,0
Exp/Cntr(USF)=0,0
Exp/Cntr=0.3,0.1

Type RM Length L Ch R = 1 ,28526   ,224.6,233.1,239.2
XS GIS Cut Line= 3
 2259651.7850175462155.7639323362259700.02390571462262.397264169
2260060.54612286462549.291704578
#Sta/Elev= 30
       0    2574    19.1 2570.34    36.7 2565.19    45.5 2561.58    67.4 2550.23
    93.7 2539.14   106.9 2537.26   136.2 2534.45   158.1 2534.29   193.9 2531.79
   215.9 2528.68   234.8  2528.4   237.1 2528.45     270 2533.28   292.8 2532.44
   312.7 2532.47   321.2 2531.87   352.6 2532.88   378.2 2532.75   398.4 2533.57
   449.5 2534.03   474.8 2534.74   487.7 2535.69   497.7 2537.39   509.1 2540.23
   531.3 2548.02   545.5 2556.18     566 2569.36   572.2 2572.43   577.8 2574.42
#Mann= 3 ,-1,0
       0      .1       0   215.9    .045       0   237.1      .1       0
#XS Ineff= 2 , 0
          158.43 2547.45
Permanent Ineff=
       F       F
Bank Sta=215.9,237.1
XS Rating Curve= 0 ,0
Exp/Cntr(USF)=0,0
Exp/Cntr=0.3,0.1

Type RM Length L Ch R = 1 ,28292   ,266.4,273,273.8
XS GIS Cut Line= 4
2259481.67946434462375.377818135 2259593.8712437462435.796595853
2259735.09696931462680.7303616812259742.91393669462742.589247151
#Sta/Elev= 30
       0 2568.07     6.1 2566.43      15  2563.1    29.1 2555.58    35.7 2552.59
    43.7 2547.56    50.9 2543.67    61.9 2538.61    68.1 2536.69    91.8  2532.6
   113.5 2532.46     129  2530.8   141.8 2531.31   152.1 2529.64     177 2529.28
   185.8 2529.62190.95372528.993   198.3 2527.86209.5987 2528.68   253.7 2531.34
   281.4  2531.1   295.2 2532.58   359.9 2531.31   376.1 2531.96   387.6 2533.09
   396.8 2536.13   410.2 2541.71   438.8 2555.73   450.9 2561.19   472.5 2569.98
#Mann= 3 ,-1,0
       0      .1       0190.9537    .045       0209.5987      .1       0
#XS Ineff= 2 , 0
          111.95 2549.12
Permanent Ineff=
       F       F
Bank Sta=190.9537,209.5987
XS Rating Curve= 0 ,0
Exp/Cntr(USF)=0,0
Exp/Cntr=0.3,0.1

Type RM Length L Ch R = 1 ,28019   ,286.6,294.4,303
XS GIS Cut Line= 2
2259342.04057742462468.0472612762259484.21835319462851.419478105
#Sta/Elev= 30
       0 2574.68    35.3 2570.01    39.6 2568.98    43.9 2566.44    55.4 2556.84
      78 2540.62    90.8 2532.48    95.1  2530.5    99.3 2529.51   107.9 2529.79
   129.2 2528.56     142 2529.03   151.9 2527.78   163.3    2527   167.6    2527
   171.9 2527.78   176.8 2528.67   184.7 2530.96   188.9 2531.26   220.4  2529.7
   235.8  2530.9   252.9 2530.99   274.2 2532.37   304.4 2532.39     334  2533.7
   341.8 2535.44   363.8 2541.92   380.9 2548.78   402.2 2559.55   408.9 2560.42
#Mann= 3 ,-1,0
       0      .1       0   151.9    .045       0   171.9      .1       0
Bank Sta=151.9,171.9
XS Rating Curve= 0 ,0
Exp/Cntr(USF)=0,0
Exp/Cntr=0.3,0.1

Type RM Length L Ch R = 1 ,27725   ,293.1,283.6,276.4
XS GIS Cut Line= 4
2259116.07946948462482.0111499692259094.40955726462823.724316545
2259097.42537493462931.8571253642259081.65833423462981.457398241
#Sta/Elev= 30
       0 2572.71     7.2 2570.56    11.2 2568.39    35.2 2553.69    51.3 2542.74
    75.3 2531.96      82 2530.41    91.4 2529.4699.298762526.917   103.4 2526.03
   110.5 2525.91   123.5 2525.97131.3983 2526.68   149.9 2527.05   175.5 2527.09
   199.6 2529.78   223.6 2529.95   270.5 2531.34   315.9 2531.81   327.8 2532.45
     375 2532.73   403.8 2533.75   431.9 2533.89   446.8 2534.62   456.2 2535.42
   460.4 2536.11   477.1 2542.05   481.5 2543.35   493.9 2548.29   502.6 2550.68
#Mann= 3 ,-1,0
       0      .1       099.29876    .045       0131.3983      .1       0
#XS Ineff= 2 , 0
                          319.28         2551.35
Permanent Ineff=
       F       F
Bank Sta=99.29876,131.3983
XS Rating Curve= 0 ,0
Exp/Cntr(USF)=0,0
Exp/Cntr=0.3,0.1

Type RM Length L Ch R = 1 ,27441   ,250.4,249.6,247
XS GIS Cut Line= 3
2258802.92018451 462530.913341672258856.92491531462739.137010776
2258831.44568693462851.676848573
#Sta/Elev= 30
       0 2589.55     6.5 2585.76    27.1 2572.85    47.8  2562.1    60.2 2556.75
    73.9 2552.24    80.9 2550.48      85 2549.83    88.2 2548.57    93.3 2545.31
   101.3 2538.51   105.6 2535.75   126.3 2525.59130.62512524.552   134.1 2524.42
153.9251 2524.49   159.4  2524.8     180 2527.51   184.2 2528.69   192.4 2532.84
   193.2 2532.96   204.8 2533.78   221.3 2535.48   241.8 2536.89   254.2 2538.66
   272.9  2539.4     291 2541.65   299.2 2543.63   319.7    2551   330.5 2553.65
#Mann= 3 ,-1,0
       0      .1       0130.6251    .045       0153.9251      .1       0
Bank Sta=130.6251,153.9251
XS Rating Curve= 0 ,0
Exp/Cntr(USF)=0,0
Exp/Cntr=0.3,0.1

Type RM Length L Ch R = 1 ,27192   ,190.1,187,185.8
XS GIS Cut Line= 2
2258548.47822596462577.931094895 2258633.1078544462828.685549529
#Sta/Elev= 30
       0 2588.99     8.6 2582.91    16.1 2578.36    20.3 2576.87    36.6 2572.99
    43.4 2570.89    46.5 2569.67      56  2565.2    62.5  2561.8    74.1 2557.51
    87.9 2555.25    92.1 2554.15   100.5 2548.16   104.7 2544.65   121.6 2526.01
   125.9 2523.93   130.1 2524.42   134.3 2524.18   138.5 2523.87     147 2523.82
   158.6 2523.93   163.9 2524.88   171.3  2526.9   176.5    2528   186.7 2531.14
   193.4 2533.82   201.8 2537.68   235.9 2549.43   260.9 2559.79   264.7 2561.03
#Mann= 3 ,-1,0
       0      .1       0   134.3    .045       0   158.6      .1       0
Bank Sta=134.3,158.6
XS Rating Curve= 0 ,0
Exp/Cntr(USF)=0,0
Exp/Cntr=0.3,0.1

Type RM Length L Ch R = 1 ,27005   ,204.6,203.3,202.2
XS GIS Cut Line= 2
2258378.55023319462682.7131833092258473.66633132462894.686201995
#Sta/Elev= 30
       0 2577.43     2.7 2576.33     7.1 2574.07    11.5 2570.95    20.2 2562.82
    30.3 2554.12    33.3 2551.28    46.5 2538.03    51.5 2533.32    55.3 2530.19
    59.7 2526.99    64.1 2524.28    68.5 2522.99    69.42522.975    90.4 2522.88
    94.1 2522.88     103 2523.08   134.2 2526.05   151.8 2528.18   156.2 2528.22
   160.5 2528.71   164.9 2529.45   166.5 2529.96   172.6 2532.34   178.1 2535.04
   193.8 2543.81   204.4 2550.17   214.9 2557.25   230.7 2566.92   232.3 2567.69
#Mann= 3 ,-1,0
       0      .1       0    69.4    .045       0    94.1      .1       0
Bank Sta=69.4,94.1
XS Rating Curve= 0 ,0
Exp/Cntr(USF)=0,0
Exp/Cntr=0.3,0.1

Type RM Length L Ch R = 1 ,26802   ,107.2,106.8,106.6
XS GIS Cut Line= 3
2258246.06709651462737.0652393832258225.00567478462834.898940314
2258300.41915258462986.405296619
#Sta/Elev= 30
       0 2568.66    16.5 2564.08    32.8  2561.1    53.3 2556.47    61.5 2554.06
    69.7 2552.42    81.9 2548.92      86 2547.06    90.1 2543.98   100.1 2539.06
   107.1 2532.74   110.1 2530.66     122 2523.63     125 2522.25   129.4 2521.86
   138.4 2521.84   144.62521.945   156.2  2522.1   172.8 2525.46   178.7 2525.38
     183 2525.84   187.7 2526.87     192 2528.41   199.6 2532.18   209.9 2538.27
   223.3 2547.23   235.4 2556.26   254.5 2569.14   263.5 2573.09   269.3  2574.6
#Mann= 3 ,-1,0
       0      .1       0     125    .045       0   144.6      .1       0
Bank Sta=125,144.6
XS Rating Curve= 0 ,0
Exp/Cntr(USF)=0,0
Exp/Cntr=0.3,0.1

Type RM Length L Ch R = 1 ,26695   ,220.3,221.3,222.4
XS GIS Cut Line= 3
2258134.31155257 462773.576736312258130.64278879462886.085492381
2258215.63581647463051.179862704
#Sta/Elev= 30
       0 2558.92    15.6 2555.63    35.6 2552.53    71.6 2546.32    83.6 2543.55
    95.7 2541.12   102.5 2538.93   107.7 2536.69   112.6 2534.07   121.9 2528.32
   129.5 2523.98     134 2522.23   138.5 2520.96     143 2520.68   156.8 2520.74
     170 2520.83   174.5 2521.76     179 2523.75   183.5 2524.58   192.5 2525.04
     197 2526.43   210.5 2534.72   220.8 2542.15   231.8 2550.87     242 2557.83
     251 2563.12   255.7 2564.99   264.5 2567.19   273.5 2568.36   298.3 2570.91
#Mann= 3 ,-1,0
       0      .1       0   138.5    .045       0   156.8      .1       0
Bank Sta=138.5,156.8
XS Rating Curve= 0 ,0
Exp/Cntr(USF)=0,0
Exp/Cntr=0.3,0.1

Type RM Length L Ch R = 1 ,26474   ,137.6,135.2,132.9
XS GIS Cut Line= 4
2257909.90550106462846.340551378 2257924.5805562462963.129531865
 2257990.0068437463106.8227801092258041.36953669463138.007272281
#Sta/Elev= 30
       0 2555.51     6.9 2552.65    10.9 2551.52    31.1 2546.86    63.3 2542.58
    90.5  2537.9   103.6  2533.8     112 2530.59   128.7 2525.98   133.1 2525.08
   149.1 2523.06   152.2 2522.45   159.5 2520.45   163.9 2519.97   164.32519.974
   188.72520.043   194.7 2520.16   209.5 2522.16     221 2523.37   225.4 2524.35
   229.8 2526.15   242.8 2533.42   245.8 2535.19   257.9 2543.21   263.9 2546.53
   269.4 2549.12   278.9 2550.21   296.4 2551.54   306.2 2552.64   335.7 2554.72
#Mann= 3 ,-1,0
       0      .1       0   164.3    .045       0   188.7      .1       0
Bank Sta=164.3,188.7
XS Rating Curve= 0 ,0
Exp/Cntr(USF)=0,0
Exp/Cntr=0.3,0.1

Type RM Length L Ch R = 1 ,26338   ,235,234.1,232.3
XS GIS Cut Line= 2
2257730.86198232462913.0800956672257911.09174659463218.687087252
#Sta/Elev= 30
       0 2551.13     9.4 2547.72    27.3  2543.3    37.3 2541.89    46.6  2541.7
    56.5 2540.89    83.7 2535.64   104.9 2528.74   111.6 2527.17   126.6 2522.09
   134.8 2521.13   148.7 2522.95   161.7 2522.91   176.3 2520.12   181.2 2519.57
     188 2519.62   211.22519.757   213.7 2519.92   220.1 2521.63   230.9 2521.95
   234.7 2522.75   237.6 2523.95   241.6  2526.9   246.2 2531.08   250.9 2534.36
   255.5 2536.27   270.3 2540.05     288 2542.61   331.1 2545.25   354.8 2547.41
#Mann= 3 ,-1,0
       0      .1       0     188    .045       0   211.2      .1       0
Bank Sta=188,211.2
XS Rating Curve= 0 ,0
Exp/Cntr(USF)=0,0
Exp/Cntr=0.3,0.1

Type RM Length L Ch R = 1 ,26104   ,326.3,322.9,326
XS GIS Cut Line= 2
2257513.01904986463030.6212462772257743.39970505463369.139760033
#Sta/Elev= 30
       0  2564.1    24.3 2555.96    55.9 2546.25    69.6 2542.39    81.8  2537.5
   104.9 2530.03   119.2 2523.36   133.6 2518.97   138.6 2518.83   148.2  2520.2
   150.9 2520.28   167.6 2519.79   182.1  2520.3   191.3  2519.3   202.32518.633
   211.4 2518.33   222.9 2518.56   225.7 2518.97   235.3 2521.37     245 2525.64
   259.5 2526.04   269.2 2526.95   275.8 2527.11   288.6 2529.79   304.2 2533.87
   312.8 2535.57     341 2538.94   366.9 2540.94   392.8 2547.64   409.5    2553
#Mann= 3 ,-1,0
       0      .1       0   202.3    .045       0   222.9      .1       0
Bank Sta=202.3,222.9
XS Rating Curve= 0 ,0
Exp/Cntr(USF)=0,0
Exp/Cntr=0.3,0.1

Type RM Length L Ch R = 1 ,25781   ,244.4,242.6,242.6
XS GIS Cut Line= 2
2257251.29408783463160.7001196182257506.75018849463496.084202692
#Sta/Elev= 30
       0 2569.96    30.8 2555.69    40.8 2551.96    55.9 2545.61    63.8 2541.26
    69.5 2537.03    74.1 2534.11   101.2 2519.74106.86642517.411   112.3 2516.03
   115.1 2515.81   123.7 2516.64   126.3 2516.76   132.3 2515.97   146.4 2518.02
   156.5 2518.38   166.5 2519.91   171.6 2520.22   195.1 2519.71   206.8 2521.04
   231.9 2521.45   240.7 2521.93   297.3 2522.08   337.8 2523.63   357.6 2524.77
   367.7 2526.17   380.6 2529.19   409.1  2537.4   417.7 2538.49   421.6 2539.41
#Mann= 3 ,-1,0
       0      .1       0106.8664    .045       0   123.7      .1       0
Bank Sta=106.8664,123.7
XS Rating Curve= 0 ,0
Exp/Cntr(USF)=0,0
Exp/Cntr=0.3,0.1

Type RM Length L Ch R = 1 ,25539   ,300.5,299,300.3
XS GIS Cut Line= 2
2257042.85444742463287.6445622772257306.14662479463618.326999326
#Sta/Elev= 30
       0 2551.08    12.2 2548.23    34.2 2539.47    47.1 2535.49    53.3 2533.25
      59 2529.84    63.3 2526.32    72.8 2519.69    78.7 2516.19    81.7 2515.52
      96 2514.74   114.4 2513.77   119.6 2514.61   130.1  2517.3   144.4 2517.89
   156.2 2517.78     170 2516.86   175.8 2517.01     186  2518.3   191.1  2518.5
   201.4 2518.35   249.7 2519.06   278.1 2518.09   324.1 2520.69   337.9 2522.42
   359.9 2528.08   380.6 2535.21   393.8 2539.31   411.9 2544.48   422.7 2546.87
#Mann= 3 ,-1,0
       0      .1       0      96    .045       0   119.6      .1       0
Bank Sta=96,119.6
XS Rating Curve= 0 ,0
Exp/Cntr(USF)=0,0
Exp/Cntr=0.3,0.1

Type RM Length L Ch R = 1 ,25240   ,291.3,313.5,335
XS GIS Cut Line= 3
2256882.99848259463339.3626685452256859.49025247463527.428509521
2257036.58558605463749.973088009
#Sta/Elev= 30
       0 2533.54     9.9 2530.35      22 2525.82      30 2523.55    50.2 2519.61
    58.3 2518.54    90.5 2518.37   110.7 2519.15     147  2517.3   165.4 2518.42
   216.9 2518.68   227.6 2517.86   239.7  2515.1   253.1 2512.79   266.72511.563
   288.9 2511.38   293.7 2511.48   304.2 2514.73   306.3 2514.88   319.6 2515.09
   333.6 2514.32   350.2 2514.34   357.6 2514.73   376.3 2514.58   404.8 2516.38
   411.6  2517.2   416.7 2518.69   437.1 2530.12   452.5 2538.23   473.9 2545.38
#Mann= 4 ,-1,0
       0      .1       0   266.7    .045       0   288.9      .1       0
  409.53     .06       0
#XS Ineff= 2 , 0
          209.84 2526.14
Permanent Ineff=
       F       F
Bank Sta=266.7,288.9
XS Rating Curve= 0 ,0
Exp/Cntr(USF)=0,0
Exp/Cntr=0.3,0.1

Type RM Length L Ch R = 1 ,24926   ,298,294.1,294.2
XS GIS Cut Line= 3
2256759.18847062463326.824945813 2256743.5163172463458.471034496
2256616.57187454463704.523843106
#Sta/Elev= 30
       0 2533.02    10.4 2527.67    14.5 2525.95    18.5 2524.74    38.6 2519.23
    51.6 2517.61    62.8 2517.16    74.9 2516.18   107.1 2516.13   144.6  2514.9
   180.6 2515.72   223.2 2514.75   243.6 2512.97   257.1  2512.3   282.6 2511.84
   288.7  2511.4   306.7 2511.83   312.2 2511.08   324.1 2507.97     336 2508.02
   342.7  2507.7   351.7 2507.91   360.7 2508.18   365.2 2509.99   378.7  2520.7
   383.2 2524.87   392.9 2534.91   396.7 2538.35   401.3 2540.68   409.4 2543.38
#Mann= 4 ,-1,0
       0      .1       0     336    .045       0   351.7      .1       0
  402.58     .06       0
Bank Sta=336,351.7
XS Rating Curve= 0 ,0
Exp/Cntr(USF)=0,0
Exp/Cntr=0.3,0.1

Type RM Length L Ch R = 1 ,24632   ,411.3,400.7,396.7
XS GIS Cut Line= 2
2256503.73236996 463259.434686132256343.87640513463613.625353301
#Sta/Elev= 30
       0 2546.56    10.7 2540.41    28.2 2529.49    45.8 2519.75    54.6 2515.81
    67.7 2511.59   121.9  2510.3   155.5 2511.54   177.5 2510.03   185.4 2507.74
   188.5  2507.3   208.2 2508.14   212.6 2507.57   215.7 2506.34   222.6 2505.08
   230.1 2504.54   247.7 2504.77   260.8 2505.55   267.1 2506.68   273.1 2507.02
   279.2 2507.11   291.6 2506.26   295.9 2506.34   304.7 2507.46   313.5 2507.39
   322.3 2508.75   333.6 2511.68     349 2517.19     379 2529.43   388.6 2533.76
#Mann= 3 ,-1,0
       0      .1       0   222.6    .045       0   247.7      .1       0
#XS Ineff= 2 , 0
          158.63 2521.18
Permanent Ineff=
       F       F
Bank Sta=222.6,247.7
XS Rating Curve= 0 ,0
Exp/Cntr(USF)=0,0
Exp/Cntr=0.3,0.1

Type RM Length L Ch R = 1 ,24231   ,327.1,320.3,316.6
XS GIS Cut Line= 4
2256111.73703898463161.9347018432256029.02192913463263.836279615
2256011.57058551463463.6963386942255997.11611257463518.972897323
#Sta/Elev= 30
       0 2534.47    14.5 2531.07      31  2526.5    44.7 2521.56    53.2 2517.39
    70.2  2504.5    75.5 2503.07    86.6 2503.86    94.5 2502.12   100.9 2502.04
   119.9 2504.51   132.6 2505.38   144.6 2504.24   168.7 2503.82   184.8 2502.16
   200.9 2503.64     233 2503.34     249 2501.66   265.1 2502.69   277.3 2501.08
   285.2 2500.62   294.6  2501.3   305.2  2503.9   321.3 2505.11   325.4 2505.92
   329.8 2507.57   341.7 2514.35   358.8 2526.31   378.9 2539.15     389 2546.46
#Mann= 3 ,-1,0
       0      .1       0   277.3    .045       0   294.6      .1       0
#XS Ineff= 2 , 0
          130.92 2514.12
Permanent Ineff=
       F       F
Bank Sta=277.3,294.6
XS Rating Curve= 0 ,0
Exp/Cntr(USF)=0,0
Exp/Cntr=0.3,0.1

Type RM Length L Ch R = 1 ,23911   ,299.6,301.5,303.7
XS GIS Cut Line= 3
2255725.13069367463054.3628966792255674.35291661 463202.88789459
2255718.78347154463526.596223369
#Sta/Elev= 30
       0 2537.76    11.4 2532.99    19.9 2530.35    36.8 2522.14    53.7 2512.56
    66.4 2504.33    78.6 2498.33    81.7 2497.72   100.2 2497.26   110.1 2499.55
   129.8 2500.69   163.3 2500.71   192.6 2496.94   207.7 2499.68   248.1 2501.01
   260.2 2498.24   280.4 2500.48   295.5 2499.28   316.7 2499.32   324.32497.743
   332.9 2496.78     345 2497.22   349.4 2498.06   381.3  2499.8   397.5 2507.51
   401.5 2510.48   417.7 2527.56   425.8  2534.6   441.9 2545.81   483.7 2572.67
#Mann= 3 ,-1,0
       0      .1       0   324.3    .045       0   349.4      .1       0
#XS Ineff= 2 , 0
          160.14  2518.5
Permanent Ineff=
       F       F
Bank Sta=324.3,349.4
XS Rating Curve= 0 ,0
Exp/Cntr(USF)=0,0
Exp/Cntr=0.3,0.1

Type RM Length L Ch R = 1 ,23610   ,237.4,231.5,228.3
XS GIS Cut Line= 4
2255365.87792095463073.4045630782255393.80569833 463199.07956131
2255415.38625359463623.0739997892255458.54736409463686.546221119
#Sta/Elev= 30
       0 2542.77    18.5 2525.94      42  2510.7    57.1 2498.42    61.2 2496.87
    73.5 2495.47   106.3 2497.46   134.8 2497.59   162.9 2494.37   190.9  2494.3
   206.9 2497.01   295.1  2497.2   315.1  2496.2   339.5 2498.26   347.1 2497.62
   350.2 2496.04   361.7 2494.42   375.2 2495.85   391.2 2497.33   407.4 2495.05
   419.2 2496.07   439.2  2495.1   463.3 2497.57   499.3 2496.05   511.3 2498.64
   523.4 2499.47   553.3 2511.13   569.8  2518.9   595.7  2533.4     630 2555.11
#Mann= 3 ,-1,0
       0      .1       0   350.2    .045       0   375.2      .1       0
#XS Ineff= 2 , 0
          130.23 2508.61
Permanent Ineff=
       F       F
Bank Sta=350.2,375.2
XS Rating Curve= 0 ,0
Exp/Cntr(USF)=0,0
Exp/Cntr=0.3,0.1

Type RM Length L Ch R = 1 ,23378   ,292.7,292.7,276.2
XS GIS Cut Line= 4
2255180.53903467463176.2295616312255152.61125728463258.743449359
2255273.20847781463639.576777335 2255344.2973657463752.557331301
#Sta/Elev= 30
       0 2545.71    26.3  2533.5    85.5 2512.28    98.1 2506.82   106.4 2501.75
     119 2496.88   142.9 2491.57     162 2492.81   177.9 2491.41     202 2495.67
     213 2494.32   219.7 2492.39   232.3  2492.6   236.5  2494.3   240.7 2495.56
   265.9 2495.72   278.5 2494.47   297.7 2495.32     354  2493.7     375 2495.27
   404.7  2493.6   425.3 2494.38   433.7  2496.3   464.7 2493.82   475.7 2496.18
   521.6 2495.83     531 2498.99   553.7 2509.35   588.5 2526.07   620.1 2543.07
#Mann= 3 ,-1,0
       0      .1       0     213    .045       0   236.5      .1       0
#XS Ineff= 2 , 0
          162.35 2508.75
Permanent Ineff=
       F       F
Bank Sta=213,236.5
XS Rating Curve= 0 ,0
Exp/Cntr(USF)=0,0
Exp/Cntr=0.3,0.1

Type RM Length L Ch R = 1 ,23085   ,317.9,349.7,378.9
XS GIS Cut Line= 4
2255121.93752488463163.648861002 2254969.4304756463386.087214484
2254951.03732942463425.1435666612255201.42486055463790.193502982
#Sta/Elev= 30
       0 2551.02    26.1 2541.66    42.6 2533.24    80.9 2516.83   103.7 2511.24
   123.2 2508.38   152.2 2506.91     191 2508.43   255.6 2507.98     276 2509.11
   299.6 2505.85   312.9 2505.25   336.1 2491.66     342 2490.17   371.5 2490.91
   379.9  2493.2   390.5 2493.76   405.1 2489.96   413.9 2491.01   463.4 2490.97
   516.6 2492.96   531.2 2491.74   555.3 2492.97   604.8 2493.04     619 2494.43
   652.4 2493.42     667 2494.04   682.6 2496.42   730.1 2507.41   755.5 2517.15
#Mann= 3 ,-1,0
       0      .1       0   336.1    .045       0   371.5      .1       0
Bank Sta=336.1,371.5
XS Rating Curve= 0 ,0
Exp/Cntr(USF)=0,0
Exp/Cntr=0.3,0.1

Type RM Length L Ch R = 1 ,22736   ,232.5,248.2,262.5
XS GIS Cut Line= 3
2255107.91782728463141.9399700992254903.39622522463435.322682021
2254624.11845137463639.844284081
#Sta/Elev= 30
       0 2552.26    23.5 2545.61    48.5 2535.99      82 2528.81   111.5 2528.13
   140.5  2523.9   188.9 2522.82   200.4 2523.76   216.4 2531.01   228.2 2531.74
   247.7  2529.3   260.7 2525.24   272.3 2526.35   286.3 2525.83   366.6 2513.56
   387.9 2508.31   409.9 2498.14   424.2 2493.63   462.3 2492.46   502.9 2494.22
   515.8 2492.82   544.4 2493.27   559.9 2492.51   573.1 2489.27   577.4 2489.26
   592.12489.389   601.7  2492.6     618 2505.34   634.3 2512.77   703.8 2552.31
#Mann= 3 ,-1,0
       0      .1       0   573.1    .045       0   592.1      .1       0
Bank Sta=573.1,592.1
XS Rating Curve= 0 ,0
Exp/Cntr(USF)=0,0
Exp/Cntr=0.3,0.1

Type RM Length L Ch R = 1 ,22488   ,183.4,184.8,186.4
XS GIS Cut Line= 3
2255103.68634586463125.0140444122254930.19560756463360.566510233
2254560.64623004463311.199226977
#Sta/Elev= 30
       0 2553.87    16.9 2546.66    44.9 2539.26    91.3 2532.03   157.1 2524.17
   208.3 2522.31   248.7 2518.65     263 2520.78   268.7 2518.82   285.9  2516.8
   292.5 2515.28   322.8 2499.39     339 2492.96   351.1 2492.11   427.8 2493.79
   443.9 2491.96   477.3 2492.28   500.3  2488.4   512.5 2488.31   521.6 2488.41
   528.8 2489.72   535.9 2492.99   560.9 2507.01   577.1 2514.69   593.2 2525.55
   605.3 2531.32   617.4 2540.93   637.6 2552.64   661.8 2573.74   665.4 2575.46
#Mann= 3 ,-1,0
       0      .1       0   500.3    .045       0   521.6      .1       0
#XS Ineff= 2 , 0
          396.39  2517.5
Permanent Ineff=
       F       F
Bank Sta=500.3,521.6
XS Rating Curve= 0 ,0
Exp/Cntr(USF)=0,0
Exp/Cntr=0.3,0.1

Type RM Length L Ch R = 1 ,22303   ,207.7,207.6,207.5
XS GIS Cut Line= 3
2255103.68634586 463099.625155882254993.66782889463201.180710007
2254621.29746376463123.603550604
#Sta/Elev= 30
       0 2557.29    14.1  2557.3    21.1 2555.89    31.8 2551.46      81 2526.02
    96.6 2520.66   111.2 2516.93   122.5 2512.67   133.8 2509.88   149.7 2504.27
   161.1 2498.49   171.7 2494.22   179.9 2491.67     189 2490.67   212.5 2491.07
   249.3 2490.31   277.9  2490.5   303.2 2492.09   359.6 2492.24   363.7 2492.14
   371.9 2489.68   383.9 2488.29   387.7 2488.16   412.7  2488.4   424.9 2489.77
   429.1 2492.02   441.3    2501   498.6 2536.81   502.6 2540.34   530.1 2559.76
#Mann= 3 ,-1,0
       0      .1       0   383.9    .045       0   412.7      .1       0
#XS Ineff= 2 , 0
          280.72  2512.2
Permanent Ineff=
       F       F
Bank Sta=383.9,412.7
XS Rating Curve= 0 ,0
Exp/Cntr(USF)=0,0
Exp/Cntr=0.3,0.1

Type RM Length L Ch R = 1 ,22095   ,233.4,218.9,207.7
XS GIS Cut Line= 3
2254997.89931031 462947.291824692254930.19560756462975.501700836
2254701.69561077462928.955405195
#Sta/Elev= 30
       0 2541.78    10.5 2541.36    19.2 2539.23    36.5 2533.15    49.5 2527.42
    58.2 2524.61    73.1  2520.8    87.7  2515.1    95.8 2512.51   116.2 2502.93
   128.5 2494.85   136.6 2490.83   140.7 2489.68   148.2 2490.78   157.1 2491.28
   177.5 2491.27   189.7 2490.46   197.9 2488.08   201.1 2487.98   214.2 2487.92
   222.12487.971   226.8 2488.34   230.5 2491.15   242.8 2501.77   250.9 2506.48
   271.4    2515   280.5 2519.51   283.6 2520.69   291.8 2525.06   306.5 2531.84
#Mann= 3 ,-1,0
       0      .1       0   201.1    .045       0   222.1      .1       0
Bank Sta=201.1,222.1
XS Rating Curve= 0 ,0
Exp/Cntr(USF)=0,0
Exp/Cntr=0.3,0.1

Type RM Length L Ch R = 1 ,21876   ,89.1,96.6,104.7
XS GIS Cut Line= 3
2254923.14313852462680.7084951082254782.09375779462754.054173088
2254710.15857362462752.643679281
#Sta/Elev= 30
       0 2506.67     7.9 2507.79    20.3 2509.24    23.3 2509.44    34.9 2509.53
    48.4 2509.02      53 2508.78    58.9 2507.86    76.7 2504.22      80 2502.58
    87.7 2495.92      89 2494.95    91.5 2493.75    93.5 2492.89   102.5 2490.15
   112.3 2487.89   122.4 2487.69   130.1 2487.89   134.1 2488.57   137.4 2489.65
   147.6 2493.65   156.8 2496.99   160.9 2499.71   176.9 2512.08   188.9    2519
   200.9 2526.45   212.9 2533.36   216.9 2536.69   221.3 2539.16   230.9 2545.49
#Mann= 3 ,-1,0
       0      .1       0   112.3    .045       0   130.1      .1       0
Bank Sta=112.3,130.1
XS Rating Curve= 0 ,0
Exp/Cntr(USF)=0,0
Exp/Cntr=0.3,0.1

Type RM Length L Ch R = 1 ,21780   ,165,175.6,186.9
XS GIS Cut Line= 3
2254900.39902685462628.8638280542254826.10656021462647.684586271
2254698.32351758462654.123266714
#Sta/Elev= 30
       0 2515.39     4.4 2515.39    13.6 2514.51    33.4 2512.02    49.7 2509.15
      58 2510.04    74.5  2510.1    78.6 2507.71    82.6 2503.23    87.5 2498.37
    91.3 2495.34    94.6 2493.32    98.6 2491.65   102.8 2490.38   118.6  2486.1
   122.6 2485.71   130.6 2485.69   134.6 2485.93   142.7 2488.13   146.7 2490.06
   150.7 2493.94   158.7 2504.23   162.7 2509.73   174.7 2527.75   182.7 2541.03
   186.7 2546.81   194.7 2556.79   198.7 2560.78   202.7 2564.27   204.6  2565.6
#Mann= 3 ,-1,0
       0      .1       0   118.6    .045       0   134.6      .1       0
Bank Sta=118.6,134.6
XS Rating Curve= 0 ,0
Exp/Cntr(USF)=0,0
Exp/Cntr=0.3,0.1

Type RM Length L Ch R = 1 ,21604   ,180.4,170.6,164.7
XS GIS Cut Line= 5
2254882.56883486462509.9958814212254831.58450023462498.008604878
2254740.57385276462474.7779215012254724.16423278462466.195573637
2254688.91313847462459.541499176
#Sta/Elev= 30
       0 2523.75    10.7  2523.4      23 2521.81    35.3  2519.3    43.5  2518.6
    51.8  2517.1    55.9 2515.81      60 2514.21    64.2 2512.17    68.3 2509.39
    72.4 2505.77    75.6 2502.57    82.2 2496.71    88.9    2491      93 2488.03
   105.4 2484.18   115.1 2483.34   121.9 2482.93   134.3 2482.83   146.8 2482.97
   151.3 2483.59   155.8  2487.2   159.6 2492.51   165.7 2500.63     176 2516.21
   179.4  2521.9   185.2 2532.52   189.2  2539.1   193.3 2543.12   200.7 2547.78
#Mann= 3 ,0,0
       0      .1       0   115.1    .045       0   151.3      .1       0
Bank Sta=115.1,151.3
XS Rating Curve= 0 ,0
Exp/Cntr(USF)=0,0
Exp/Cntr=0.3,0.1

Type RM Length L Ch R = 1 ,21433   ,239.1,236.1,234.3
XS GIS Cut Line= 3
2254929.12433319462306.3454290982254790.44506212462357.854872639
2254723.08655903462342.005813088
#Sta/Elev= 30
       0 2524.16     9.5  2520.7    18.1 2518.27    26.6 2514.84    30.9 2512.62
    43.7 2502.54    52.2  2493.7    56.5 2488.24    60.8 2483.34      65 2480.45
    73.6 2477.43    78.82476.204    82.1  2475.6    86.4 2475.44    90.6 2475.75
    94.9  2476.5     112 2477.51   116.2 2478.24   120.5  2479.1   133.6 2483.07
   137.6 2483.54   141.8 2484.68   146.1 2487.54   150.1 2491.14   166.2 2506.39
   170.8 2510.26   191.4  2523.4   199.6 2527.45   203.6 2529.88   217.1 2536.83
#Mann= 3 ,-1,0
       0      .1       0    78.8    .045       0    94.9      .1       0
Bank Sta=78.8,94.9
XS Rating Curve= 0 ,0
Exp/Cntr(USF)=0,0
Exp/Cntr=0.3,0.1

Type RM Length L Ch R = 1 ,21197   ,138.5,140.8,143.2
XS GIS Cut Line= 2
2254832.77263165462075.5481797012254649.51788059462180.107947573
#Sta/Elev= 30
       0 2515.78    10.4  2514.6    19.2 2514.73    28.3 2513.95    42.1 2511.22
    46.7 2509.52    51.5 2506.37      56 2501.78    63.2 2493.42    66.1 2490.33
    69.1 2487.78    74.4 2483.88      79 2479.06    80.8 2478.06    83.6 2477.13
    88.2 2476.34    97.4 2471.49   103.3 2470.23   113.1 2469.81   121.1 2470.05
     125 2470.39   129.6  2473.4   130.7 2474.38   132.4 2476.22   157.3 2506.94
   161.9 2511.68   171.1 2519.23   179.5 2524.62   184.9 2527.42     211 2539.38
#Mann= 3 ,-1,0
       0      .1       0   103.3    .045       0   121.1      .1       0
Bank Sta=103.3,121.1
XS Rating Curve= 0 ,0
Exp/Cntr(USF)=0,0
Exp/Cntr=0.3,0.1

Type RM Length L Ch R = 1 ,21057   ,224.7,221.9,219.4
XS GIS Cut Line= 3
 2254777.4256173461989.2660345352254726.47584367461984.451882697
2254571.08962474462046.272869758
#Sta/Elev= 30
       0 2511.27    17.3 2509.61    21.3 2508.97    29.4 2507.41    37.4 2505.12
    41.4 2504.65    45.5 2503.77    49.5 2502.33    53.7  2499.4    62.7 2488.87
    65.8 2485.89    70.9 2481.63    75.2 2478.67    79.5 2476.19    93.5 2469.04
    96.7 2467.54    99.7 2466.72   105.3 2465.95   108.9 2466.91     112 2469.24
   122.5 2478.23   131.1 2483.39   139.7 2496.96   142.8 2500.76   148.4 2504.98
   152.7  2507.3   169.9 2513.19   187.1 2520.17   195.7  2523.2   218.4 2533.29
#Mann= 3 ,-1,0
       0      .1       0    99.7    .045       0   108.9      .1       0
Bank Sta=99.7,108.9
XS Rating Curve= 0 ,0
Exp/Cntr(USF)=0,0
Exp/Cntr=0.3,0.1

Type RM Length L Ch R = 1 ,20835   ,194.6,193,192.4
XS GIS Cut Line= 4
2254800.13771933461613.4638587542254769.96373468461624.813155329
2254655.00913608461762.3917972662254480.24808302461866.853568288
#Sta/Elev= 30
       0 2489.98       6 2486.77    17.1 2478.36    32.2 2467.98      35  2466.7
    41.3 2464.73    50.8 2463.21    78.7 2463.03   142.2 2466.38   181.4 2466.18
   224.1 2467.25   230.2 2466.82   238.1 2464.21   242.8 2463.36 285.7952463.348
     294 2462.52   298.7 2462.65303.09492463.545     309 2465.44   331.3 2467.31
     336 2469.31   341.7  2473.8   358.5 2491.96   370.2 2503.76   373.1 2506.32
   382.6 2511.96   391.9 2519.92   396.5 2522.59   402.3 2526.88   415.1  2534.5
#Mann= 3 ,-1,0
       0      .1       0 285.795    .045       0303.0949      .1       0
#XS Ineff= 2 , 0
          212.85  2477.6
Permanent Ineff=
       F       F
Bank Sta=285.795,303.0949
XS Rating Curve= 0 ,0
Exp/Cntr(USF)=0,0
Exp/Cntr=0.3,0.1

Type RM Length L Ch R = 1 ,20642   ,275.4,274.1,272.9
XS GIS Cut Line= 3
2254673.01310354461443.1914514512254551.59835127461600.750269214
2254375.87154128461710.288755676
#Sta/Elev= 30
       0 2489.34    32.8 2477.11    47.6 2467.34    63.1 2458.97    88.4 2458.12
   104.7 2459.77     139 2459.16   178.8 2462.03   193.1 2463.77   204.6  2463.5
   224.9 2457.99   235.9 2457.65238.5577 2457.68264.74992458.201   278.4 2461.84
   303.3 2460.75   313.1 2459.13   320.9 2461.25   335.3 2462.89   341.1 2464.49
   346.9 2468.14     351 2472.32   353.8 2477.24   358.5 2487.72   363.2 2494.75
     373 2501.22   381.7  2508.2   391.5 2514.31   400.9 2521.62     406 2524.47
#Mann= 3 ,-1,0
       0      .1       0238.5577    .045       0264.7499      .1       0
#XS Ineff= 2 , 0
          193.78  2476.6
Permanent Ineff=
       F       F
Bank Sta=238.5577,264.7499
XS Rating Curve= 0 ,0
Exp/Cntr(USF)=0,0
Exp/Cntr=0.3,0.1

Type RM Length L Ch R = 1 ,20368   ,267,273.4,278.9
XS GIS Cut Line= 3
2254533.04038493461273.1611751912254373.95038574461388.869773983
2254237.93731453461483.704031928
#Sta/Elev= 30
       0 2477.39      11 2471.31    23.5 2466.52    27.2 2465.39    35.7 2464.12
    47.6 2460.98    55.5 2457.95    65.4 2452.27    70.3  2451.2    75.1 2450.96
    88.4 2453.09   124.7  2452.1   159.3 2454.41   198.2 2455.64   206.8 2455.18
   218.2 2452.42228.60352452.032   251.62451.925     272 2452.12   281.5 2453.45
   290.2 2453.89   296.4 2455.13   301.3 2457.81   310.3 2465.58   315.9 2471.23
   318.9 2475.98   327.5 2487.27   335.4 2496.85   344.7 2506.87   362.5 2519.68
#Mann= 3 ,-1,0
       0      .1       0228.6035    .045       0   251.6      .1       0
Bank Sta=228.6035,251.6
XS Rating Curve= 0 ,0
Exp/Cntr(USF)=0,0
Exp/Cntr=0.3,0.1

Type RM Length L Ch R = 1 ,20094   ,292.4,289.7,285.3
XS GIS Cut Line= 3
2254458.09782064461038.0890977872254225.94313389461178.722657489
2254108.98003374461211.121058381
#Sta/Elev= 30
       0 2508.61     6.6 2504.39    12.4  2499.6      21  2496.2    29.9  2490.7
    39.7 2482.99      60 2464.17    73.5  2453.1    77.1 2450.45    86.4 2447.14
    95.8 2446.34   105.1 2447.82   123.1 2448.97   175.3 2448.28   198.7 2450.27
     225 2449.58   236.6 2450.06   259.5 2448.74   273.3 2450.05   281.4 2449.61
304.47052445.896   310.6 2445.78319.0827 2445.83   327.2 2445.87   331.4 2447.07
   335.5 2449.61   343.8 2457.42   372.9 2475.97   385.3 2488.16   392.8 2494.07
#Mann= 3 ,-1,0
       0      .1       0304.4705    .045       0319.0827      .1       0
Bank Sta=304.4705,319.0827
XS Rating Curve= 0 ,0
Exp/Cntr(USF)=0,0
Exp/Cntr=0.3,0.1

Type RM Length L Ch R = 1 ,19804   ,348.9,358.3,364.7
XS GIS Cut Line= 2
2254323.68327041460810.393706609    2253975.2913460989.526420138
#Sta/Elev= 30
       0 2483.93     8.4 2479.79    21.9 2472.02    52.2 2460.53    58.6 2456.57
    67.3  2449.1    71.4 2446.38      76  2444.2    80.4  2442.8    89.4 2441.32
    98.4 2440.77   116.4 2441.24   125.4 2442.38   159.1 2444.03   174.9 2443.91
   210.8 2446.45   230.4  2444.4   246.8 2444.22   251.2 2443.53   260.1    2445
   264.8 2445.04   283.9 2444.16   303.5 2444.09   309.8 2443.28   318.8 2442.63
     321 2443.87   332.3 2448.15   355.2 2472.29     373 2485.87   391.7 2498.31
#Mann= 3 ,-1,0
       0      .1       0   309.8    .045       0     321      .1       0
Bank Sta=309.8,321
XS Rating Curve= 0 ,0
Exp/Cntr(USF)=0,0
Exp/Cntr=0.3,0.1

Type RM Length L Ch R = 1 ,19446   ,374.6,378.2,374.2
XS GIS Cut Line= 3
2254257.12302269 460599.161974172254192.24030755460603.393455592
2253849.49031237 460614.67740605
#Sta/Elev= 30
       0 2475.76      13 2471.34      33 2462.83    61.1 2446.96    69.1 2443.37
    77.1 2440.54    97.1 2437.98   117.2 2436.18   129.1 2434.25   153.1 2433.44
   165.1 2435.94   181.1 2436.57   205.2 2435.23   233.2 2436.98   241.2 2436.72
   255.72434.816   277.2 2434.73   286.92435.636   293.2 2437.97   301.2 2439.06
   321.2 2437.97   329.2 2436.98   341.2 2437.87   345.8 2440.33   349.7 2443.17
   357.1 2450.11   365.2 2458.58   373.6 2464.97   397.3 2479.02     408 2483.67
#Mann= 3 ,-1,0
       0      .1       0   255.7    .045       0   286.9      .1       0
#XS Ineff= 2 , 0
                          300.28         2443.79
Permanent Ineff=
       F       F
Bank Sta=255.7,286.9
XS Rating Curve= 0 ,0
Exp/Cntr(USF)=0,0
Exp/Cntr=0.3,0.1

Type RM Length L Ch R = 1 ,19068   ,102.7,99.9,102.2
XS GIS Cut Line= 2
2254267.89766186 460264.761987462253817.42934231460300.202559184
#Sta/Elev= 30
       0 2462.21    11.8 2457.65    19.8 2455.45    35.8 2453.24      80 2443.83
      84 2441.75      96    2432    99.4 2430.17   112.5  2427.7   120.1 2426.91
   140.2 2427.66   152.2 2430.13   160.1  2430.5   188.3 2428.24   208.4 2428.61
   228.4 2432.44   240.5 2433.46   252.5 2432.16   284.6 2433.58   296.6 2432.86
   308.7 2433.17   324.7  2428.7   343.3 2429.94   378.1 2430.48   384.9 2431.78
   396.9  2439.4     401  2442.7   409.3 2450.92     425 2463.99   451.9 2480.88
#Mann= 3 ,0,0
       0      .1       0   112.5    .045       0   140.2      .1       0
#XS Ineff= 2 , 0
                          367.11         2440.49
Permanent Ineff=
       F       F
Bank Sta=112.5,140.2
XS Rating Curve= 0 ,0
Exp/Cntr(USF)=0,0
Exp/Cntr=0.3,0.1

Type RM Length L Ch R = 1 ,18968   ,279.4,279.5,280.4
XS GIS Cut Line= 2
 2254302.5258633 460158.745567632253841.29438831460208.112850886
#Sta/Elev= 30
       0 2465.57    18.5  2458.9    30.5 2453.71    50.6 2447.48    94.9 2436.06
     119  2432.2   131.1 2426.02   147.2 2425.47     157 2425.71   183.4  2428.4
   215.6  2426.8   229.7  2428.6   243.7 2426.97   263.8 2426.96   275.9 2425.66
     286 2426.59   300.1 2429.59   316.1 2430.28   320.2  2430.3   328.2 2428.66
   348.3 2427.93   360.4 2426.59   364.8 2426.65   380.5 2429.45   412.7 2429.34
   416.7 2430.72   423.4 2434.86     444 2452.52   456.9  2462.3   463.9 2466.61
#Mann= 3 ,-1,0
       0      .1       0   131.1    .045       0     157      .1       0
#XS Ineff= 2 , 0
                           380.4         2437.68
Permanent Ineff=
       F       F
Bank Sta=131.1,157
XS Rating Curve= 0 ,0
Exp/Cntr(USF)=0,0
Exp/Cntr=0.3,0.1

Type RM Length L Ch R = 1 ,18689   ,232.1,231.1,230.5
XS GIS Cut Line= 2
2254315.22030757459941.5295213042253869.50426446459949.992484148
#Sta/Elev= 30
       0 2449.23      19 2440.45    31.1 2437.19    51.1 2433.37    75.1 2431.04
    99.1 2429.21   127.1 2428.93   143.1 2427.51   163.1 2427.95   175.1 2427.09
   191.1 2426.97   199.1 2426.03   207.1 2423.23   211.1 2422.73   227.1 2424.58
   251.1 2424.99   255.1  2424.8   263.1  2423.2   287.1 2422.24   293.2 2421.38
   303.1 2420.77   313.4 2421.41   331.1 2425.69   351.1 2425.94   367.1 2424.49
   387.1 2427.74   399.2 2434.01     411 2441.03   435.1 2456.93   445.8 2464.81
#Mann= 3 ,-1,0
       0      .1       0   293.2    .045       0   313.4      .1       0
Bank Sta=293.2,313.4
XS Rating Curve= 0 ,0
Exp/Cntr(USF)=0,0
Exp/Cntr=0.3,0.1

Type RM Length L Ch R = 1 ,18457   ,269.7,247.7,230.7
XS GIS Cut Line= 4
2254358.36323063459763.822780253 2254224.9487039459704.566561675
2253918.87154771459721.4924873632253832.77531529459771.163539519
#Sta/Elev= 30
       0 2444.61      33 2435.94    54.9 2433.62    75.5 2432.87    95.2 2430.99
   124.8 2430.82   174.8 2427.94   206.8 2427.56     214 2426.87   222.5 2424.63
   238.9 2422.07   294.6 2422.56     319  2421.6     327 2419.77     335 2418.79
   347.1 2420.02   359.1 2419.99   367.1 2419.07   386.5 2419.42   407.2 2419.54
   423.2 2420.47   435.2  2419.3   443.2 2422.43   447.2 2423.16   474.8 2422.14
   492.6 2422.51   497.2 2423.35   504.1 2426.21   511.1 2430.31   551.9 2460.22
#Mann= 3 ,-1,0
       0      .1       0   359.1    .045       0   386.5      .1       0
Bank Sta=359.1,386.5
XS Rating Curve= 0 ,0
Exp/Cntr(USF)=0,0
Exp/Cntr=0.3,0.1

Type RM Length L Ch R = 1 ,18210   ,331.2,336,344.1
XS GIS Cut Line= 4
2254120.34520663459260.2998297022253957.72881231459469.576235954
2253936.66739058459515.0960829162253765.36800846 459700.55721936
#Sta/Elev= 30
       0 2441.68     6.4 2439.49    36.6 2433.64      67 2425.34    82.2 2423.49
    92.3 2424.15   106.2 2421.77   168.3 2420.47   228.8 2419.66     269 2420.25
   273.4    2420   282.2 2415.55     290 2415.36   305.1  2415.6   323.5 2417.61
   345.4  2417.5   361.6  2416.3   386.7 2417.51   398.4    2417   404.3 2415.09
   421.5 2414.89   426.9 2415.61   432.4 2418.86   437.8 2419.91     465  2418.3
   486.8 2419.18   515.2 2421.88   530.4 2428.54     552 2441.07   567.7  2451.4
#Mann= 3 ,-1,0
       0      .1       0     290    .045       0   305.1      .1       0
#XS Ineff= 2 , 0
          269.28 2430.14
Permanent Ineff=
       F       F
Bank Sta=290,305.1
XS Rating Curve= 0 ,0
Exp/Cntr(USF)=0,0
Exp/Cntr=0.3,0.1
