HEC-RAS study THRNYCK.prj: THRNYCK

--- THRNYCK.g01 (geometry) --- (continued)

Type RM Length L Ch R = 1 ,17874   ,133.4,134.5,137.2
XS GIS Cut Line= 2
2253865.40500751459114.3281102182253521.75272616459607.079302632
#Sta/Elev= 30
       0 2449.47    11.6 2442.86    37.1 2419.62    42.5 2417.65    57.1 2415.16
    96.1 2414.05   109.2 2415.76     121 2414.69     140 2415.71   169.3 2415.08
   218.9 2416.51     250 2414.73   261.9 2415.76   266.8 2414.87     273 2412.15
   286.3 2413.23     301 2411.21   316.8  2413.8   362.1 2413.53     379 2414.84
   434.12409.458   442.4 2408.47   456.7 2408.53     4612409.489   471.6 2414.97
   474.1 2415.38   525.3 2416.53   549.7 2421.06   569.2 2427.03   600.8 2440.24
#Mann= 3 ,-1,0
       0      .1       0   434.1    .045       0     461      .1       0
#XS Ineff= 2 , 0
          262.15 2426.75
Permanent Ineff=
       F       F
Bank Sta=434.1,461
XS Rating Curve= 0 ,0
Exp/Cntr(USF)=0,0
Exp/Cntr=0.3,0.1

Type RM Length L Ch R = 1 ,17739   ,259.2,261.3,263
XS GIS Cut Line= 4
2253682.55973263459067.6764485112253642.06189359459244.570694561
 2253451.6452296459463.1972346942253420.61436584459583.089208316
#Sta/Elev= 30
       0 2433.66     9.7 2426.73    28.6 2414.76    38.5 2410.82    79.5 2411.92
   108.2  2411.3   163.5  2414.5   181.5 2414.76   187.6 2413.86   197.4 2409.49
   202.6 2409.12   245.2 2412.36   257.4 2411.71   277.8 2412.74   288.4 2411.53
   302.3 2413.67   320.2 2411.55   367.5 2412.98   378.9 2408.94   394.5 2409.55
401.55292409.032     421  2408.3 426.2532408.935   436.9 2413.15   442.2 2414.32
   495.6 2414.05   531.3 2414.96   556.1  2422.3   571.1 2428.71   595.2 2440.63
#Mann= 3 ,-1,0
       0      .1       0401.5529    .045       0 426.253      .1       0
#XS Ineff= 2 ,-1
       0  173.49 2423.95  442.77     594 2419.94
Permanent Ineff=
       F       F
Bank Sta=401.5529,426.253
XS Rating Curve= 0 ,0
Exp/Cntr(USF)=0,0
Exp/Cntr=0.3,0.1

Type RM Length L Ch R = 1 ,17478   ,321.1,312.3,294.9
XS GIS Cut Line= 4
2253441.77177295459020.3021791982253410.74090919459126.089214746
2253229.03174505459318.6882540592253161.99597319459516.198687932
#Sta/Elev= 30
       0 2438.14    21.8 2435.81    30.1 2433.52    34.3 2429.89    38.4 2425.34
    55.1 2408.67    59.3 2407.38    82.6 2407.38   117.1 2409.55   136.5 2407.79
     153 2407.87   169.5 2405.97     186  2406.6   213.1 2408.65     230 2406.96
     248 2407.61   264.2 2406.66   281.2 2406.93   290.5 2406.55   323.72406.902
   341.3 2408.69     353 2408.91   367.5 2410.27   399.7 2409.54   453.7 2409.97
   500.2 2412.71   508.6 2414.15   521.3 2418.29   555.1 2433.28   583.6 2447.37
#Mann= 3 ,-1,0
       0      .1       0   281.2    .045       0   323.7      .1       0
#XS Ineff= 2 ,-1
   29.52   124.1 2416.62  370.48   567.1 2416.75
Permanent Ineff=
       F       F
Bank Sta=281.2,323.7
XS Rating Curve= 0 ,0
Exp/Cntr(USF)=0,0
Exp/Cntr=0.3,0.1

Type RM Length L Ch R = 1 ,17166   ,315.1,312.2,309.1
XS GIS Cut Line= 3
  2253104.663753458977.9873649782253063.75943259 459229.05526268
2252996.05572984459415.240445245
#Sta/Elev= 30
       0 2450.44     7.3 2447.14    13.7 2442.83    27.6 2430.78    31.6 2425.47
    35.7 2421.59    47.8 2413.96    55.9 2404.52      60 2401.61      64  2400.6
    68.1 2400.43    88.3 2401.04    97.3 2403.03   111.2  2404.4   132.9  2402.4
   145.1 2404.25   157.2 2403.84     174 2402.75   189.7  2400.7   205.3 2400.69
   226.2  2405.6   246.4 2407.54   284.3 2406.13   322.6 2405.98   358.5 2406.96
   365.2 2406.59     395 2407.08   399.2 2407.76   407.1 2410.53   452.5 2432.27
#Mann= 3 ,-1,0
       0      .1       0      60    .045       0    88.3      .1       0
#XS Ineff= 2 , 0
                          252.01         2417.14
Permanent Ineff=
       F       F
Bank Sta=60,88.3
XS Rating Curve= 0 ,0
Exp/Cntr(USF)=0,0
Exp/Cntr=0.3,0.1

Type RM Length L Ch R = 1 ,16853   ,339.7,338.3,337.1
XS GIS Cut Line= 2
2252784.48165874458932.8515631442252774.60820209459419.471926667
#Sta/Elev= 30
       0 2446.48    16.3 2433.81    28.3 2426.25    44.3 2412.34    59.4 2400.93
    72.3 2396.06    76.3 2395.43    88.3 2395.44    92.3 2395.88   104.3 2398.24
   132.4 2397.84   156.4 2396.78   164.4 2397.42   172.4 2397.08   176.4 2397.36
   196.4 2401.29   204.4 2402.35   216.4 2403.03   228.4 2402.74   244.4 2401.29
   284.4 2401.49   304.4 2400.89   320.4    2401   336.4  2402.3   404.4 2403.63
   408.4 2404.31   420.2 2407.84     432 2412.39   455.5    2423   486.7  2439.1
#Mann= 3 ,-1,0
       0      .1       0    72.3    .045       0    92.3      .1       0
#XS Ineff= 2 , 0
                          220.88         2412.11
Permanent Ineff=
       F       F
Bank Sta=72.3,92.3
XS Rating Curve= 0 ,0
Exp/Cntr(USF)=0,0
Exp/Cntr=0.3,0.1

Type RM Length L Ch R = 1 ,16515   ,315.7,304.7,291.2
XS GIS Cut Line= 2
2252440.32116976458938.4935383742252467.12055209 459460.37624708
#Sta/Elev= 30
       0 2444.85    26.7  2432.7    30.7 2429.32    38.7 2420.61    46.7 2413.18
    54.8 2408.03    74.8 2391.28    78.8 2389.69   106.8  2389.5   114.8 2389.91
   118.8 2390.51   126.9 2393.44   142.9 2393.91   162.9 2393.15   186.9 2393.41
     223 2397.52     239 2397.43   279.1  2394.3   287.1 2395.05   295.1 2397.08
   327.1 2398.05   367.2 2396.25   395.2  2396.3   423.2 2397.45   439.3 2400.35
   451.3 2403.79   463.4 2408.57   475.9 2414.21   491.3 2422.38   522.6 2440.65
#Mann= 3 ,-1,0
       0      .1       0    78.8    .045       0   114.8      .1       0
#XS Ineff= 2 , 0
                           225.3         2408.07
Permanent Ineff=
       F       F
Bank Sta=78.8,114.8
XS Rating Curve= 0 ,0
Exp/Cntr(USF)=0,0
Exp/Cntr=0.3,0.1

Type RM Length L Ch R = 1 ,16210   ,254.3,266.4,282.2
XS GIS Cut Line= 4
2252140.96461169458977.1485986812252134.01811396459082.367395964
2252201.36602533459206.7177946792252207.20272447459440.358805745
#Sta/Elev= 30
       0 2407.38    12.1 2404.63    44.1 2400.63    56.2 2397.49    76.2 2394.25
   120.9 2390.96139.53842387.147     145 2386.14   154.1 2385.77   167.8 2386.01
173.03792387.194   181.4 2388.92   199.6 2388.94   204.2 2388.76   213.3 2386.83
   217.8 2386.53   222.4 2388.04   231.5 2393.16   254.7 2394.36   277.3 2393.17
   317.3 2393.49   349.6 2392.85     373 2390.73   397.4 2389.77   404.3 2390.11
   413.4 2391.51   429.4 2395.46   437.4  2398.2   453.4 2405.94   480.6  2422.5
#Mann= 3 ,-1,0
       0      .1       0139.5384    .045       0173.0379      .1       0
#XS Ineff= 2 , 0
                          347.89          2403.8
Permanent Ineff=
       F       F
Bank Sta=139.5384,173.0379
XS Rating Curve= 0 ,0
Exp/Cntr(USF)=0,0
Exp/Cntr=0.3,0.1

Type RM Length L Ch R = 1 ,15944   ,368.4,366,363
XS GIS Cut Line= 2
2251898.69154775459006.197241125 2251908.5650044459456.144765658
#Sta/Elev= 30
       0 2423.67      27 2419.44      39 2415.18      47 2409.66      63 2396.49
      79 2387.32      83 2386.22      87 2385.99      95 2387.12     147 2387.95
     167  2383.9     203 2383.35   211.9 2384.42     223 2385.84     235 2385.31
     251 2383.19   255.2 2384.01     267 2388.78     271 2389.05   331.1 2389.28
   339.1 2388.42   351.1 2384.86   355.1 2384.55   373.8 2385.51   379.1 2386.73
   395.1 2394.67   415.5 2409.44   419.1 2412.67   427.2 2423.47   450.1  2442.9
#Mann= 3 ,-1,0
       0      .1       0     167    .045       0   211.9      .1       0
#XS Ineff= 2 , 0
          132.03 2401.35  322.79         2399.47
Permanent Ineff=
       F       F
Bank Sta=167,211.9
XS Rating Curve= 0 ,0
Exp/Cntr(USF)=0,0
Exp/Cntr=0.3,0.1

Type RM Length L Ch R = 1 ,15578   ,294.2,293.9,284.5
XS GIS Cut Line= 2
2251513.62673835458989.2713154372251562.99402161 459454.73427185
#Sta/Elev= 30
       0  2421.7    36.1 2400.82    44.2 2396.66    64.3  2383.7    68.3 2381.45
    72.3 2380.52    84.4 2379.83   100.4 2381.81   108.5 2380.64   124.6 2382.46
   140.7 2382.26   172.9 2383.13     201 2382.83   205.1 2382.16   209.1 2380.36
   213.1 2379.59   245.3 2379.59   251.7 2380.14   261.4 2382.05   281.5 2379.74
   289.5 2381.28   305.6 2381.28   317.7 2380.95   333.8  2378.3   337.8 2378.59
   349.9 2377.71   353.9 2378.05   357.9 2380.11   386.1 2398.24   468.1 2456.51
#Mann= 3 ,-1,0
       0      .1       0   209.1    .045       0   251.7      .1       0
#XS Ineff= 2 , 0
          153.61 2396.25
Permanent Ineff=
       F       F
Bank Sta=209.1,251.7
XS Rating Curve= 0 ,0
Exp/Cntr(USF)=0,0
Exp/Cntr=0.3,0.1

Type RM Length L Ch R = 1 ,15284   ,283.3,276.2,268.1
XS GIS Cut Line= 3
2251276.01837395459052.6534502082251268.32484657459199.524979285
2251318.74227741459461.786740887
#Sta/Elev= 30
       0 2413.69    16.5 2407.54    28.6 2401.79    40.6 2394.64    60.6 2380.54
    64.6 2379.25    72.6 2377.78    96.7 2377.82   110.7  2376.6   116.7 2376.67
   124.7 2375.73   136.7 2375.49   144.7 2377.49   152.8 2378.25   177.3 2378.28
   199.6 2379.02   213.9 2378.74   226.1 2377.59   238.4 2378.83   250.9 2377.82
   258.7 2375.17     285 2373.71   291.3 2373.38   311.7 2373.44316.27642374.685
   319.8 2377.58   332.1 2390.19   348.3 2401.95   361.1 2410.79   414.1 2444.94
#Mann= 3 ,-1,0
       0      .1       0     285    .045       0316.2764      .1       0
#XS Ineff= 2 , 0
           100.4  2395.4
Permanent Ineff=
       F       F
Bank Sta=285,316.2764
XS Rating Curve= 0 ,0
Exp/Cntr(USF)=0,0
Exp/Cntr=0.3,0.1

Type RM Length L Ch R = 1 ,15008   ,363.7,363.1,363.1
XS GIS Cut Line= 2
2250895.83045075459162.7620537362251093.29958377459537.953406482
#Sta/Elev= 30
       0 2413.43     7.3 2409.79    11.8 2408.87    34.6 2393.86    52.5  2383.8
      66 2377.36    73.1 2375.04    84.1 2374.35    93.1 2372.75   102.7 2373.13
   117.5  2371.7   133.8 2372.12   147.2 2374.45   160.9 2374.18   170.9 2374.96
   209.3  2373.8   232.6 2374.48   256.7 2371.38   284.2 2370.05   309.9 2369.88
     316 2370.45   319.1 2370.98   323.7 2373.83   333.7 2384.32   350.8 2397.53
   378.2 2415.28   395.9 2427.85   404.8 2433.34   409.5 2437.15     424 2446.51
#Mann= 3 ,-1,0
       0      .1       0   284.2    .045       0     316      .1       0
Bank Sta=284.2,316
XS Rating Curve= 0 ,0
Exp/Cntr(USF)=0,0
Exp/Cntr=0.3,0.1

Type RM Length L Ch R = 1 ,14645   ,323.3,325.8,327.9
XS GIS Cut Line= 2
2250577.05885029 459344.715754882250774.52798332459702.981181937
#Sta/Elev= 30
       0 2418.67     9.7 2415.22    23.4 2407.07    32.5  2402.2    46.2 2396.85
    64.5  2386.9    73.3 2383.63    79.2 2380.76    85.1 2377.24    96.4 2369.44
     101 2368.18   110.1 2367.82   126.3 2365.55     141 2365.31     165 2367.77
   192.4 2368.71   206.1 2367.94   217.1 2366.68   233.5 2367.26   246.8 2366.53
   274.6 2366.59   283.7 2367.46   292.8 2367.53     302  2369.6   305.9 2371.22
   320.2 2381.25   329.4 2386.31   341.2 2393.92   367.7 2409.81   409.1 2432.89
#Mann= 3 ,-1,0
       0      .1       0   246.8    .045       0   274.6      .1       0
Bank Sta=246.8,274.6
XS Rating Curve= 0 ,0
Exp/Cntr(USF)=0,0
Exp/Cntr=0.3,0.1

Type RM Length L Ch R = 1 ,14319   ,296.4,312.8,332
XS GIS Cut Line= 2
2250310.47552071459460.3762470792250472.68230855459859.545994549
#Sta/Elev= 30
       0 2404.39     5.2 2401.98    13.8 2396.19    41.8 2379.94    61.3 2364.93
    78.6 2360.22    82.9 2359.76      91 2360.66   104.5 2363.54   126.1 2364.34
     137 2363.19   147.7 2363.55   161.6 2360.52   169.3 2360.89   177.9 2363.55
   186.5 2364.11   195.2 2363.96   199.5 2363.02   203.8 2360.96   229.7 2363.96
   238.4 2363.53   262.9 2364.37     282 2362.81     302 2362.91   308.9 2363.62
   318.1 2365.87   346.3 2368.36   354.8 2369.96   372.2 2376.65   430.9 2393.47
#Mann= 3 ,-1,0
       0      .1       0     282    .045       0     302      .1       0
Bank Sta=282,302
XS Rating Curve= 0 ,0
Exp/Cntr(USF)=0,0
Exp/Cntr=0.3,0.1

Type RM Length L Ch R = 1 ,14006   ,340.9,341.3,341.2
XS GIS Cut Line= 4
2250184.94157186459485.765135611 2250173.6576214459626.814516342
2250079.15453631459784.7898227622250077.74404251459893.397845925
#Sta/Elev= 30
       0 2405.27    11.5 2401.29    19.5 2396.62    39.5 2382.29    59.6 2366.34
    63.6 2363.67    67.6 2361.75   107.8 2355.54   111.8 2355.72   119.8 2357.58
   127.8 2357.18   144.3    2359     156  2359.3   181.5 2358.19   191.1 2360.26
   214.2 2361.16   223.5 2360.82   231.8 2359.47   240.5 2358.95   246.8 2358.42
     258 2358.98   270.1 2360.87   279.4  2360.8   302.7 2362.82     370 2361.69
     386 2364.83     402 2369.67     414 2374.71     426 2378.69   434.2 2382.21
#Mann= 3 ,-1,0
       0      .1       0   240.5    .045       0     258      .1       0
#XS Ineff= 2 , 0
                          322.79          2371.8
Permanent Ineff=
       F       F
Bank Sta=240.5,258
XS Rating Curve= 0 ,0
Exp/Cntr(USF)=0,0
Exp/Cntr=0.3,0.1

Type RM Length L Ch R = 1 ,13665   ,258.1,278.5,295.7
XS GIS Cut Line= 4
2250009.18956759459409.3173658942249894.06727232459449.727367285
2249778.45239211459640.7221232032249657.04520289459696.552899921
#Sta/Elev= 30
       0 2382.62    10.1 2379.43    44.6 2370.39    73.7 2364.49   101.1  2360.6
   115.5 2357.54   128.8 2357.22   141.1 2354.03   148.8 2353.34   157.9 2353.54
   175.4 2355.07   191.5 2353.37   210.2 2353.16   213.3 2352.68   219.6 2351.86
   228.9 2352.56   247.6 2355.73   289.7 2355.63   312.3 2354.42   326.5 2357.08
   347.8 2357.94   369.8  2357.2   387.4 2355.12   400.6 2355.15   410.7 2354.18
   414.2 2355.14     427 2362.29   453.4 2381.15   461.3 2385.48   478.9 2397.56
#Mann= 3 ,-1,0
       0      .1       0   213.3    .045       0   228.9      .1       0
#XS Ineff= 2 , 0
          130.52    2371  355.42         2367.12
Permanent Ineff=
       F       F
Bank Sta=213.3,228.9
XS Rating Curve= 0 ,0
Exp/Cntr(USF)=0,0
Exp/Cntr=0.3,0.1

Type RM Length L Ch R = 1 ,13386   ,291.1,297.2,302.3
XS GIS Cut Line= 4
2249986.41334442459297.8666276792249903.54724126459300.409883691
2249805.79028716 459339.701875662249548.80886476459343.305261072
#Sta/Elev= 30
       0 2390.15    70.3 2363.47    82.3 2360.64    92.2 2357.34   103.8 2355.38
     123 2353.73   203.1 2355.48   217.9 2353.87   233.9 2349.91   265.9 2351.08
   277.7 2350.77   301.9 2352.44   313.9 2351.21321.86312348.779   329.9 2347.88
339.26282348.472   345.9 2349.82   353.9 2349.56   357.9 2350.18   361.9 2353.82
   365.9 2360.66     371 2371.22   377.9  2386.9   381.9 2394.05   385.9 2398.85
   405.9 2416.64   421.9 2437.31   429.9 2446.32   437.9 2458.02   445.3 2463.75
#Mann= 3 ,-1,0
       0      .1       0321.8631    .045       0339.2628      .1       0
#XS Ineff= 2 , 0
          125.42 2372.44
Permanent Ineff=
       F       F
Bank Sta=321.8631,339.2628
XS Rating Curve= 0 ,0
Exp/Cntr(USF)=0,0
Exp/Cntr=0.3,0.1

Type RM Length L Ch R = 1 ,13089   ,170,168.1,166.6
XS GIS Cut Line= 4
2249919.24701805459039.6843615162249786.21907355459069.432735372
2249681.83926765459039.6099336852249599.64737281459039.350176982
#Sta/Elev= 30
       0 2377.27    44.1 2357.69    52.3 2355.22    68.7 2352.25      81 2349.22
    97.4 2348.42   109.7 2349.12   117.9 2348.96   130.2 2351.27   134.3 2351.38
   138.4    2351   142.6 2350.08   150.9 2346.98   167.6 2347.93   175.9 2346.91
   180.2 2345.65187.72522345.111210.17612344.488   213.3 2344.46   217.5 2344.67
   234.1 2349.03   243.8 2356.27   258.5 2369.36   266.5 2375.67   278.5 2383.93
   294.5 2396.68   298.5 2400.19   302.5 2404.36   318.5 2417.98   327.1 2425.75
#Mann= 3 ,-1,0
       0      .1       0187.7252    .045       0210.1761      .1       0
#XS Ineff= 2 , 0
           80.81  2366.1
Permanent Ineff=
       F       F
Bank Sta=187.7252,210.1761
XS Rating Curve= 0 ,0
Exp/Cntr(USF)=0,0
Exp/Cntr=0.3,0.1

Type RM Length L Ch R = 1 ,12921   ,188.7,185.3,182
XS GIS Cut Line= 4
2249932.53719433458883.0402248282249798.33458674458895.155738013
2249741.48487102458883.972187381 2249647.3566532458898.883588224
#Sta/Elev= 30
       0 2391.41     9.7 2386.22    24.5 2377.31    40.5 2368.66    83.3 2347.25
    88.7 2344.61    92.7 2342.99    96.8 2343.01   100.8 2343.44   108.8 2343.09
   112.8 2343.28   120.9 2344.81   136.9 2345.52   153.3 2343.96   158.7 2342.96
   161.4  2342.6   165.5 2342.56   178.32342.663   206.2  2343.8   218.3 2345.83
   222.9  2345.9   230.5 2345.51   234.5 2345.73   250.6 2347.85   254.8 2348.94
   258.8 2351.18   262.9 2354.44   275.3 2365.94   283.1 2373.99     288 2378.12
#Mann= 3 ,-1,0
       0      .1       0   158.7    .045       0   178.3      .1       0
Bank Sta=158.7,178.3
XS Rating Curve= 0 ,0
Exp/Cntr(USF)=0,0
Exp/Cntr=0.3,0.1

Type RM Length L Ch R = 1 ,12736   ,175.9,161.3,148
XS GIS Cut Line= 4
2249913.89794328458691.0559389682249858.91215267458714.355002786
2249790.87888632458710.6271525752249605.41833833458769.340793396
#Sta/Elev= 30
       0 2397.51    14.9 2390.08    27.9 2381.87      41 2372.57    62.5 2356.27
    66.5 2352.56    74.5 2343.61    78.5 2340.84    82.5 2339.94    86.72339.835
   102.5 2339.44   110.72339.714   122.5 2341.31   135.2 2344.36   160.1 2345.54
   185.2 2345.14   193.6  2345.9   214.6 2345.52     223 2346.14   239.8 2346.09
   252.4 2344.41   265.9 2341.51   269.1 2341.22   272.3 2341.78   277.5 2344.32
   297.8 2358.66   302.7 2363.66   311.1 2375.71   315.3 2378.97   322.4 2381.91
#Mann= 3 ,-1,0
       0      .1       0    86.7    .045       0   110.7      .1       0
Bank Sta=86.7,110.7
XS Rating Curve= 0 ,0
Exp/Cntr(USF)=0,0
Exp/Cntr=0.3,0.1

Type RM Length L Ch R = 1 ,12574   ,276.9,270.9,266.1
XS GIS Cut Line= 2
2249828.80386124458517.5371769262249548.25664297458700.337174354
#Sta/Elev= 30
       0 2391.82    10.3 2386.18    29.1 2371.23    43.7 2356.28    53.3 2347.76
      58 2342.63    62.8 2341.27    72.6 2341.24      84 2339.91    91.5 2338.96
     113 2339.53   131.2 2340.04   139.2 2341.95   153.2 2342.78   163.1 2344.13
   196.8 2345.54   208.3 2345.52   231.5 2344.16   244.2 2342.15     249 2342.12
   257.5 2340.26   263.2 2340.43   266.1 2340.98   268.1 2341.72   282.4  2352.6
   287.2 2355.39     292  2359.1   300.8 2370.17   303.7 2372.52   334.8 2392.11
#Mann= 3 ,-1,0
       0      .1       0      84    .045       0     113      .1       0
Bank Sta=84,113
XS Rating Curve= 0 ,0
Exp/Cntr(USF)=0,0
Exp/Cntr=0.3,0.1

Type RM Length L Ch R = 1 ,12303   ,339.9,339.5,342.2
XS GIS Cut Line= 2
2249640.92608611458295.3844022742249421.31220031458531.501065619
#Sta/Elev= 30
       0 2387.39    21.6 2372.38    29.8 2366.07    35.8 2360.98    48.1 2349.02
    51.6 2346.44    59.8 2339.33    62.5 2337.48    65.7 2336.38    77.5 2335.49
   100.8    2335   106.2 2334.97   123.5 2336.51     139 2335.13   147.9 2335.29
   171.4 2339.19   185.8 2339.97   214.1 2339.22     221 2338.47   228.2  2336.7
   231.1  2336.6     236 2337.07   242.8  2339.1   259.2 2340.35   265.4 2342.35
   270.7 2344.75   287.7 2354.48   301.8 2363.15   313.8 2371.27   322.5 2376.03
#Mann= 3 ,-1,0
       0      .1       0    77.5    .045       0   100.8      .1       0
Bank Sta=77.5,100.8
XS Rating Curve= 0 ,0
Exp/Cntr(USF)=0,0
Exp/Cntr=0.3,0.1

Type RM Length L Ch R = 1 ,11964   ,189.5,188.8,188.6
XS GIS Cut Line= 2
2249381.23883174458152.3654395182249158.92890897458359.310965509
#Sta/Elev= 30
       0  2362.3     6.9 2359.55    12.6 2357.86    24.7 2351.77    35.3 2347.89
    42.3 2343.92    60.8 2336.96      78 2337.06    83.4 2336.28    97.6 2333.05
   108.9 2331.83   132.6 2332.03   154.5 2330.47   165.6 2329.56   171.4 2329.68
   176.3 2330.63   183.2 2333.78   188.1 2334.57   203.7 2334.38   212.5 2331.86
   219.3 2331.68   224.3 2332.35     236 2334.99   241.9 2337.19   253.6 2345.27
   264.5 2354.61   277.1 2363.99   292.8 2377.06   296.6 2380.72   303.7 2386.22
#Mann= 3 ,-1,0
       0      .1       0   154.5    .045       0   176.3      .1       0
Bank Sta=154.5,176.3
XS Rating Curve= 0 ,0
Exp/Cntr(USF)=0,0
Exp/Cntr=0.3,0.1

Type RM Length L Ch R = 1 ,11775   ,334,345.7,359
XS GIS Cut Line= 2
2249261.36220256458005.9510730142249030.32331693458226.834403239
#Sta/Elev= 30
       0 2375.95    29.3 2361.38    33.6 2359.93    40.4 2358.47      57 2350.82
      71 2346.53    90.2 2338.79   102.1 2334.73   116.3 2334.73   128.9  2334.1
   137.8 2330.84   143.6 2329.81   158.7 2331.01   175.7 2328.89   184.1  2328.5
   189.8 2328.97   198.3  2328.7   218.8 2328.62   235.1 2329.43   237.9 2330.09
   239.6 2330.96   252.1 2339.37   257.7 2343.56   265.1 2350.47   271.9 2355.85
   278.3 2362.34   289.4 2372.17   299.9 2379.91   311.5 2387.59   319.6 2392.46
#Mann= 3 ,-1,0
       0      .1       0   198.3    .045       0   218.8      .1       0
Bank Sta=198.3,218.8
XS Rating Curve= 0 ,0
Exp/Cntr(USF)=0,0
Exp/Cntr=0.3,0.1

Type RM Length L Ch R = 1 ,11430   ,409.9,412,414.5
XS GIS Cut Line= 2
2249159.54179155457811.3558803632248862.49179573457862.768379639
#Sta/Elev= 30
       0 2365.46     7.5 2363.37    14.9 2360.81    28.7 2355.25      44 2349.74
    76.5 2338.58    88.7 2334.89   104.9 2331.03   117.1 2328.84   125.2  2329.4
   137.4 2329.54   149.6 2330.45   156.8 2330.11   163.7 2328.61   169.9 2326.15
   174.9 2324.54     178 2323.98   189.52323.565   198.3 2323.25   214.5 2323.38
   222.6 2323.78     226 2324.31   230.7 2326.13   238.9 2332.36   246.7  2339.5
   255.1 2346.49   259.2 2350.18     264 2355.35   275.4 2366.27   301.5 2387.11
#Mann= 3 ,-1,0
       0      .1       0   189.5    .045       0   214.5      .1       0
#XS Ineff= 2 , 0
          151.46 2343.45
Permanent Ineff=
       F       F
Bank Sta=189.5,214.5
XS Rating Curve= 0 ,0
Exp/Cntr(USF)=0,0
Exp/Cntr=0.3,0.1

Type RM Length L Ch R = 1 ,11018   ,309.4,308.6,307.1
XS GIS Cut Line= 2
2249109.27179226457422.9058858292248824.78929626457442.328385556
#Sta/Elev= 30
       0 2349.18    21.1 2340.86    29.2 2337.38    36.9 2334.63    53.2 2331.53
    65.2 2329.99      82 2328.32   101.3 2327.65   113.4  2327.6   117.4 2326.91
   121.4 2325.56   133.4 2324.43   141.4 2322.74   161.5 2319.69   169.5 2319.06
   180.72318.995   197.6 2318.72   205.3 2318.89   213.6 2318.95   217.6 2320.25
   221.6 2322.75   229.6 2328.72   241.7 2336.05   245.7  2338.8   249.7 2341.05
   253.7 2345.85   257.7 2351.54   265.5 2361.65   269.6 2366.42   285.1 2377.88
#Mann= 3 ,-1,0
       0      .1       0   180.7    .045       0   205.3      .1       0
Bank Sta=180.7,205.3
XS Rating Curve= 0 ,0
Exp/Cntr(USF)=0,0
Exp/Cntr=0.3,0.1

Type RM Length L Ch R = 1 ,10709   ,191.8,173.2,149.6
XS GIS Cut Line= 3
2249032.72429334457113.2883901862248824.78929626457137.280889848
2248763.09429713457248.103388289
#Sta/Elev= 30
       0 2367.79     7.6 2360.22    16.7 2353.86    36.8  2335.3    44.8 2329.66
    52.9 2323.02    54.5 2322.25      61  2319.9      65 2319.01    85.1 2319.15
   109.3  2316.3   117.3 2316.11   137.5 2315.97   145.5 2316.16   153.6 2316.42
   169.7 2321.06   173.7 2321.79   185.8  2323.3   201.9 2324.04   218.5 2323.64
     242 2324.08   277.3 2320.93   282.4 2321.08   290.1 2324.06     295 2326.69
   314.5 2340.71   319.1 2343.34   323.6 2347.62   332.8 2357.68   336.2  2359.9
#Mann= 3 ,-1,0
       0      .1       0   117.3    .045       0   145.5      .1       0
#XS Ineff= 2 , 0
                          193.27         2336.17
Permanent Ineff=
       F       F
Bank Sta=117.3,145.5
XS Rating Curve= 0 ,0
Exp/Cntr(USF)=0,0
Exp/Cntr=0.3,0.1

Type RM Length L Ch R = 1 ,10536   ,171.1,158.7,143
XS GIS Cut Line= 3
2248867.79083752456909.634628688 2248798.0983385457131.279625569
2248739.83083932457248.957123913
#Sta/Elev= 30
       0 2383.88    20.5 2365.65    37.3 2349.51    41.5 2344.69    52.1 2331.25
    62.4 2317.36    65.4 2315.02    66.6 2314.06    70.8  2313.7    79.1 2314.59
    98.2 2316.89   108.5 2317.38   130.1 2319.51   133.7 2319.63   150.5 2318.34
     162  2318.8   171.4 2321.73     184 2323.14   225.9 2322.25   252.3 2323.49
   270.2  2321.8   283.6  2321.3   292.5 2320.42   301.4 2322.55   305.9 2324.19
   323.7 2334.85   337.1 2344.54   346.1 2354.65   350.5 2358.92   363.7 2363.73
#Mann= 3 ,-1,0
       0      .1       0    65.4    .045       0    79.1      .1       0
#XS Ineff= 2 , 0
                          197.59         2334.66
Permanent Ineff=
       F       F
Bank Sta=65.4,79.1
XS Rating Curve= 0 ,0
Exp/Cntr(USF)=0,0
Exp/Cntr=0.3,0.1

Type RM Length L Ch R = 1 ,10377   ,173.1,174.1,181
XS GIS Cut Line= 4
2248687.85031268 456901.262484062248688.35616187456995.096447288
2248728.60827899457061.2798200262248721.97715331457235.704526929
#Sta/Elev= 30
       0 2362.49    19.9 2347.24    27.9 2340.47    35.9 2333.25    47.9 2321.41
    55.9 2316.28    59.9 2315.16    71.9 2314.85    83.9 2312.7793.246482311.976
   124.4 2312.09   139.7  2311.8   152.5 2312.49   166.5 2316.24   171.3 2316.26
   187.2 2314.65   191.2 2315.07   199.2 2317.71   211.2 2318.18   227.2 2320.03
   251.3 2320.72   279.6 2319.57   287.3 2319.84   291.2 2320.52   295.3 2322.19
   298.9 2324.39   303.3 2328.29   311.3 2336.17   339.3  2355.9   345.8 2359.39
#Mann= 3 ,-1,0
       0      .1       093.24648    .045       0   124.4      .1       0
#XS Ineff= 2 , 0
                          172.67         2320.39
Permanent Ineff=
       F       F
Bank Sta=93.24648,124.4
XS Rating Curve= 0 ,0
Exp/Cntr(USF)=0,0
Exp/Cntr=0.3,0.1

Type RM Length L Ch R = 1 ,10203   ,277,266.4,256.3
XS GIS Cut Line= 2
2248530.75334226456910.7771286722248575.31084164457243.244623994
#Sta/Elev= 30
       0 2360.53     6.5 2355.92    14.1 2349.09    18.6  2343.8    30.7 2334.09
    50.9 2319.86    58.9  2315.1      63 2313.44      71 2312.22    91.2 2312.46
    95.9 2311.63   103.3  2309.3   107.4 2308.84   115.4 2309.94   127.5 2310.39
   151.7 2309.56   173.6  2310.6   188.5 2309.57   206.3 2309.57   213.4 2311.12
   228.4 2317.67   244.6 2318.14   264.7 2317.79   270.3 2318.59   280.9 2322.94
   294.7 2333.31   305.1 2340.38   309.1 2342.58     318 2346.64   335.4 2353.39
#Mann= 3 ,-1,0
       0      .1       0   188.5    .045       0   206.3      .1       0
Bank Sta=188.5,206.3
XS Rating Curve= 0 ,0
Exp/Cntr(USF)=0,0
Exp/Cntr=0.3,0.1

Type RM Length L Ch R = 1 ,9937    ,205.4,206,207.2
XS GIS Cut Line= 2
2248269.12084594457006.7471273222248422.21584379457318.649622933
#Sta/Elev= 30
       0 2352.68     2.7  2349.4     4.1 2348.24    16.1 2340.06      25 2334.68
    29.4 2331.22    33.9 2326.64      40 2317.73    42.8 2314.13    45.9 2312.01
    54.9 2306.84    60.6 2304.82    79.6  2304.1    90.8 2304.44   100.7 2306.45
   114.1 2307.66   140.8 2308.97   154.2 2309.08   165.5 2308.65   167.6 2308.87
     172 2311.28   176.5 2313.01   185.4 2313.81   216.3 2314.26   237.2 2314.13
   256.7  2313.3   282.1 2314.44   287.9 2315.81   323.5 2330.05   347.4 2337.44
#Mann= 3 ,-1,0
       0      .1       0    60.6    .045       0    90.8      .1       0
Bank Sta=60.6,90.8
XS Rating Curve= 0 ,0
Exp/Cntr(USF)=0,0
Exp/Cntr=0.3,0.1

Type RM Length L Ch R = 1 ,9731    ,184.2,199.5,218.9
XS GIS Cut Line= 2
2248093.13316023457105.2576728572248229.88053484457422.209736298
#Sta/Elev= 30
       0  2345.4    11.4  2335.9    26.6 2319.95    34.8 2312.48    39.1 2308.08
    41.8 2306.11    47.8 2303.12    65.3 2302.29    90.5 2302.63    95.8 2303.03
   100.1  2304.5   104.5 2307.05   105.7 2307.19     135 2306.42   156.7 2308.43
   165.5 2307.48   169.6 2307.47   181.8 2309.73   191.6 2310.46   204.7 2310.64
   219.7 2310.19   229.8 2311.06   246.9 2311.53   261.3 2312.64   265.7 2313.41
   276.2 2316.46   309.2 2327.33   322.3 2330.48   339.7 2336.81   345.2  2338.4
#Mann= 3 ,-1,0
       0      .1       0    65.3    .045       0    90.5      .1       0
#XS Ineff= 2 , 0
                          156.98         2308.17
Permanent Ineff=
       F       F
Bank Sta=65.3,90.5
XS Rating Curve= 0 ,0
Exp/Cntr(USF)=0,0
Exp/Cntr=0.3,0.1

Type RM Length L Ch R = 1 ,9531    ,139.3,156,176.2
XS GIS Cut Line= 3
2248050.74782132457068.1757906622247956.24473623457116.132580111
2247822.24782453457464.524550517
#Sta/Elev= 30
       0 2348.15     7.4  2344.6    43.3 2322.93    55.3 2314.73    65.7 2306.65
    74.7 2305.11   111.4 2304.76   125.4 2301.18   158.5 2300.82   165.6 2299.91
   175.7 2299.19   190.4 2299.81   201.4  2301.8   224.5 2300.76   244.2 2300.85
   257.1 2303.99   261.4 2304.29   312.8 2301.84   325.7 2302.96   334.2 2302.51
   347.1 2303.25   364.2  2302.4   368.5 2303.53   377.1 2307.55   394.2 2317.85
   419.9 2336.33   432.8 2344.34   453.5 2352.28   462.8  2354.5   479.2 2359.93
#Mann= 3 ,-1,0
       0      .1       0   165.6    .045       0   190.4      .1       0
#XS Ineff= 2 , 0
          109.94 2312.81  261.04          2315.9
Permanent Ineff=
       F       F
Bank Sta=165.6,190.4
XS Rating Curve= 0 ,0
Exp/Cntr(USF)=0,0
Exp/Cntr=0.3,0.1

Type RM Length L Ch R = 1 ,9375    ,146.3,149.9,156.7
XS GIS Cut Line= 3
2248045.10584609457055.4813463972247943.55029196457062.533815433
2247595.15832155457165.499863367
#Sta/Elev= 30
       0 2346.85       9 2342.25      25 2332.22      33  2327.9    57.1 2308.93
    65.1 2304.31    73.1 2303.82    81.2 2302.43   105.3 2303.23     122 2302.66
   130.3 2301.96   138.7 2300.19   151.7 2299.24   180.4 2299.38   209.6 2297.65
     229 2297.94   243.82297.208   254.7 2296.51   264.4  2296.9     293  2297.1
   312.7 2298.02   326.4 2297.08   355.6  2297.1   363.9 2298.98   372.3 2303.42
   379.3 2309.16   405.6 2334.69   426.5 2353.87   443.2 2365.26   465.1  2378.7
#Mann= 3 ,-1,0
       0      .1       0   243.8    .045       0   264.4      .1       0
Bank Sta=243.8,264.4
XS Rating Curve= 0 ,0
Exp/Cntr(USF)=0,0
Exp/Cntr=0.3,0.1

Type RM Length L Ch R = 1 ,9225    ,139,148.8,162.6
XS GIS Cut Line= 3
2248044.90341435456996.3677383542247940.17633441456958.864774337
2247664.27251811  456959.5677675
#Sta/Elev= 30
       0 2335.91    21.8 2318.75    30.5 2314.68    43.7 2305.19    47.5  2303.4
    53.1 2302.17    60.3 2301.09    77.3 2301.05    98.5 2299.58   115.2 2300.93
   123.2 2300.72   139.2 2298.67   159.2 2299.39   175.2  2296.9   187.2 2297.39
   195.2 2297.05   203.2 2296.33   211.2 2294.85223.28822294.439   231.2 2294.36
249.1882 2294.49   267.2 2296.54   299.2 2295.72   311.2 2294.51   319.2 2295.42
   331.2 2301.31   339.2 2307.01     345 2312.33   363.2 2330.93   387.1 2348.61
#Mann= 3 ,-1,0
       0      .1       0223.2882    .045       0249.1882      .1       0
#XS Ineff= 2 , 0
          120.08  2315.2
Permanent Ineff=
       F       F
Bank Sta=223.2882,249.1882
XS Rating Curve= 0 ,0
Exp/Cntr(USF)=0,0
Exp/Cntr=0.3,0.1

Type RM Length L Ch R = 1 ,9076    ,130.7,130.5,130.1
XS GIS Cut Line= 2
2248053.87576584456952.3410364682247748.19204855456765.948525923
#Sta/Elev= 30
       0 2327.54      16 2316.31    25.4 2311.87    39.5 2303.47    48.8 2299.62
    53.5 2299.24    62.9 2299.45    72.3 2298.35    81.6 2298.85   109.7    2298
   123.8 2298.42   142.5 2296.89   154.9 2296.74   161.3 2295.91   170.7  2296.5
     180  2296.4   189.8 2295.95   236.2 2292.16   245.1 2292.37   262.6 2291.87
   282.7  2291.5   285.8 2291.86   297.1 2294.51   300.4 2296.16   306.5 2299.88
     312 2305.13   314.9 2309.13   329.9 2328.11   339.3 2337.98     358 2354.61
#Mann= 3 ,0,0
       0      .1       0   262.6    .045       0   285.8      .1       0
#XS Ineff= 2 , 0
           125.3  2307.5
Permanent Ineff=
       F       F
Bank Sta=262.6,285.8
XS Rating Curve= 0 ,0
Exp/Cntr(USF)=0,0
Exp/Cntr=0.3,0.1

Type RM Length L Ch R = 1 ,8946    ,178.7,178.8,178.4
XS GIS Cut Line= 2
2248136.78794356456850.9597443372247809.55338027456652.080117506
#Sta/Elev= 30
       0 2347.91    33.5 2322.38    45.4 2311.93    57.3 2303.63    66.2 2298.24
    70.9 2296.16    74.5 2295.36    80.3 2294.91   129.8 2295.78   147.3 2295.37
   167.7  2293.6   180.6 2294.72   193.9 2294.95     202 2294.21   208.5 2292.77
   220.7 2294.13   242.2 2293.96   265.3 2289.96   276.9 2289.34   298.7 2289.07
   303.8 2289.52   309.7 2290.71   314.3  2293.5     319 2298.03   333.6 2315.46
   342.4 2324.69     350 2331.44   356.5 2336.31   365.8 2345.17   382.9 2359.06
#Mann= 3 ,-1,0
       0      .1       0   276.9    .045       0   303.8      .1       0
#XS Ineff= 2 , 0
           128.4 2299.13
Permanent Ineff=
       F       F
Bank Sta=276.9,303.8
XS Rating Curve= 0 ,0
Exp/Cntr(USF)=0,0
Exp/Cntr=0.3,0.1

Type RM Length L Ch R = 1 ,8767    ,244.9,243.7,245
XS GIS Cut Line= 2
2248203.82931047456686.1968899082247919.26696839456510.383700751
#Sta/Elev= 30
       0 2318.57       9 2312.97    32.5 2296.92      40  2292.9    46.6 2291.17
    64.4  2291.5    74.8 2292.51    84.2 2292.46   102.2 2293.68   125.5 2293.24
   154.8 2294.61   164.2 2294.21   169.1 2293.51   178.3 2290.34   206.5 2291.42
     215 2289.52   225.3 2288.02     230 2287.84   258.2    2288     265 2288.87
   273.7 2292.85   275.9  2294.6   281.7 2301.29   291.1  2309.6   295.8 2314.31
   302.7  2322.8   306.3  2327.8   319.3 2340.03   329.2 2347.55   334.5  2352.3
#Mann= 3 ,0,0
       0      .1       0   225.3    .045       0   258.2      .1       0
#XS Ineff= 2 , 0
          154.14  2297.4
Permanent Ineff=
       F       F
Bank Sta=225.3,258.2
XS Rating Curve= 0 ,0
Exp/Cntr(USF)=0,0
Exp/Cntr=0.3,0.1

Type RM Length L Ch R = 1 ,8524    ,215.8,215.1,214.6
XS GIS Cut Line= 2
2248314.61816026456460.1931347242248073.56326196456325.948683299
#Sta/Elev= 30
       0 2318.47       7 2314.84    16.5 2308.89    21.1 2306.89    30.5 2301.68
    34.8 2299.84      44 2296.56    59.9 2293.07    71.6 2289.07    74.6 2288.44
    89.8 2286.47    95.2 2286.96   118.7 2287.51   140.2  2287.3   149.3 2288.83
   153.9 2288.77   156.9 2288.09   172.2 2285.88   183.4 2285.69   192.2 2285.87
     218 2286.86   227.1 2286.59   230.4 2287.41   233.4  2288.7   239.3 2291.91
   245.5 2294.61     250 2297.02     254 2299.77   271.6 2312.92   275.9 2315.57
#Mann= 3 ,-1,0
       0      .1       0   172.2    .045       0   192.2      .1       0
Bank Sta=172.2,192.2
XS Rating Curve= 0 ,0
Exp/Cntr(USF)=0,0
Exp/Cntr=0.3,0.1

Type RM Length L Ch R = 1 ,8308    ,164.9,164.2,163.5
XS GIS Cut Line= 3
2248400.14482576456256.9208635162248171.24536475456141.337967362
2248063.97235002 456154.18051138
#Sta/Elev= 30
       0 2325.98     5.7 2321.67    17.7 2314.27    31.3 2302.29    40.3 2295.68
    47.4 2288.77    53.7 2283.67    58.2 2282.45    62.7 2282.36    71.7 2282.93
    94.1 2285.82     103 2284.71   116.5 2284.42   125.4 2283.49   141.4 2285.04
   151.6 2283.34   185.62283.174   197.1 2282.96   211.2 2286.67     224 2285.73
     233 2286.35   246.4 2285.99   255.4 2289.45   263.5 2289.84   275.6 2294.96
   291.7 2298.64   299.8 2299.65   344.1  2300.1   352.2 2301.12   364.5 2303.75
#Mann= 3 ,0,0
       0      .1       0   151.6    .045       0   185.6      .1       0
Bank Sta=151.6,185.6
XS Rating Curve= 0 ,0
Exp/Cntr(USF)=0,0
Exp/Cntr=0.3,0.1

Type RM Length L Ch R = 1 ,8144    ,337.8,323.6,307.5
XS GIS Cut Line= 3
2248432.94262251456087.5216213042248193.40007837455972.998362023
2248070.50724664455993.847978375
#Sta/Elev= 30
       0 2309.79    14.7 2299.49    20.3 2294.35    27.5 2286.78    31.9  2283.9
    45.2 2282.55    54.1 2280.55    62.3 2280.06    71.3 2280.47    76.2 2282.07
    80.3 2282.54      94 2281.79   107.3 2281.85118.43912280.789147.49892280.686
   163.1 2283.03   188.3 2280.72   195.9 2282.66   200.4 2283.18   218.1 2282.25
   235.8 2280.35   240.3 2281.78   244.7 2284.51   249.1 2286.12   266.8 2286.09
   280.6  2287.5   311.4  2287.4   343.8  2294.3   353.4  2295.3   390.2 2297.03
#Mann= 3 ,-1,0
       0      .1       0118.4391    .045       0147.4989      .1       0
Bank Sta=118.4391,147.4989
XS Rating Curve= 0 ,0
Exp/Cntr(USF)=0,0
Exp/Cntr=0.3,0.1

Type RM Length L Ch R = 1 ,7821    ,304.7,324.8,334.5
XS GIS Cut Line= 3
2248471.55767822455736.1461866372248423.60088877455720.630754756
2248034.41587938455791.158012604
#Sta/Elev= 30
       0 2343.02     7.8 2338.96    22.6 2327.66      33 2320.97    44.1 2312.12
    57.3 2303.71    66.1 2295.75    74.2 2287.35    82.3 2280.04    86.4 2277.56
88.282952276.969    94.5 2276.15115.85222276.259   155.5 2277.12   171.8 2275.05
     184  2277.2   207.9 2275.97   216.5 2277.32   224.6 2277.54   236.8 2279.01
     249 2278.41   261.2 2281.68   277.8 2284.55   305.9 2285.25   318.8 2284.43
   342.5 2284.51   366.9 2286.12   399.4 2286.37   423.8 2287.91   445.9 2290.91
#Mann= 3 ,-1,0
       0      .1       088.28295    .045       0115.8522      .1       0
Bank Sta=88.28295,115.8522
XS Rating Curve= 0 ,0
Exp/Cntr(USF)=0,0
Exp/Cntr=0.3,0.1

Type RM Length L Ch R = 1 ,7496    ,357.4,380.2,406.3
XS GIS Cut Line= 4
2248557.59780046455654.3375458132248464.50520918455513.288165082
 2248275.9811711455434.2435501532248150.33703104455278.024292463
#Sta/Elev= 30
       0 2315.31    44.5  2287.9    56.7 2282.53    73.3  2277.4    82.9 2275.78
   111.6 2274.44   120.2 2273.24   140.4 2275.31   182.4 2275.59   199.7 2274.83
   212.1  2271.4   224.3 2270.85   242.7 2273.02   273.2 2272.61   297.7  2273.5
   319.1 2271.91   348.7 2271.91   360.2 2275.03   376.9 2275.73   405.6 2272.16
   436.4 2272.94   449.7 2272.68   462.5 2271.29   477.5 2272.93   499.2 2273.65
   503.1 2275.14   518.5 2286.37   533.9 2295.67   550.4 2305.05   573.9  2316.8
#Mann= 3 ,0,0
       0      .1       0   319.1    .045       0   348.7      .1       0
#XS Ineff= 2 , 0
          179.52 2284.25
Permanent Ineff=
       F       F
Bank Sta=319.1,348.7
XS Rating Curve= 0 ,0
Exp/Cntr(USF)=0,0
Exp/Cntr=0.3,0.1

Type RM Length L Ch R = 1 ,7116    ,258.8,263.1,273.8
XS GIS Cut Line= 3
2248709.93113165455616.2542130152248603.14102904455246.902004544
2248588.13229131 455161.91026241
#Sta/Elev= 30
       0 2319.23    28.2 2301.61    65.7  2281.7    82.3 2273.73    94.3 2271.17
   115.6 2271.54   119.8 2271.03   128.1 2268.05   140.6 2267.41   161.4    2269
   211.4 2269.77   215.6 2269.26   223.9 2265.89     228  2265.5   248.9 2267.55
   265.5 2267.59   273.9 2265.54   307.2 2267.57   319.7 2266.39     353 2267.73
   365.7 2266.41   386.2 2268.07   395.4 2265.34   405.8 2264.96   410.6 2264.74
     435 2264.95   447.2 2268.58   455.3 2275.36   459.3 2279.72   470.8 2300.66
#Mann= 3 ,0,0
       0      .1       0   405.8    .045       0     435      .1       0
#XS Ineff= 2 , 0
          201.81 2279.95
Permanent Ineff=
       F       F
Bank Sta=405.8,435
XS Rating Curve= 0 ,0
Exp/Cntr(USF)=0,0
Exp/Cntr=0.3,0.1

Type RM Length L Ch R = 1 ,6853    ,192.6,173.1,160.7
XS GIS Cut Line= 4
2248920.28395591455463.2926813512248841.64533356455374.870113438
2248863.61662529455212.500967896 2248833.8141368455175.143927136
#Sta/Elev= 30
       0 2297.78    21.4 2286.97    32.7 2281.86    54.3 2270.74    61.7 2267.37
    69.6 2265.25    75.2 2264.91     120 2267.74   124.1 2267.59     136 2264.94
   140.2 2264.43   156.4 2265.28   180.6 2265.51   184.6 2264.97   196.7 2261.81
   207.4 2261.74   212.9  2261.8   216.9 2262.57233.3183 2261.98261.45422261.994
   269.4 2262.48   273.4 2263.55   281.5 2264.45   286.4 2264.51   296.7 2263.71
   301.8 2264.36   306.9 2265.87   309.8 2268.28   315.5 2274.63     330 2294.08
#Mann= 3 ,-1,0
       0      .1       0233.3183    .045       0261.4542      .1       0
#XS Ineff= 2 , 0
          120.53  2276.9
Permanent Ineff=
       F       F
Bank Sta=233.3183,261.4542
XS Rating Curve= 0 ,0
Exp/Cntr(USF)=0,0
Exp/Cntr=0.3,0.1

Type RM Length L Ch R = 1 ,6680    ,359.8,330.2,308.2
XS GIS Cut Line= 4
2249148.77122388455375.9635314862249096.40643486455349.670883434
2248960.32925122455144.3604483252248849.32338858455124.331436261
#Sta/Elev= 30
       0 2334.64    41.3 2311.31    68.8  2296.9    97.6 2280.89     114 2271.18
   122.6 2266.94   128.4 2264.61   134.2 2263.11   155.2 2261.56   164.8 2259.54
   169.6 2258.99   189.3 2259.51   203.1 2261.13   217.5 2262.08   232.8 2261.38
   254.5 2261.38   270.3 2259.36   281.3 2259.97   298.7 2261.97   325.4 2260.72
   341.6 2258.68   345.7 2259.15   353.8  2261.9   357.9    2265   370.1 2277.42
   375.5 2282.37   382.3 2286.74   398.5 2298.32   410.7 2305.99   417.7 2309.34
#Mann= 3 ,-1,0
       0      .1       0   164.8    .045       0   189.3      .1       0
Bank Sta=164.8,189.3
XS Rating Curve= 0 ,0
Exp/Cntr(USF)=0,0
Exp/Cntr=0.3,0.1

Type RM Length L Ch R = 1 ,6349    ,376,362.9,347.4
XS GIS Cut Line= 3
2249272.16491727454965.0126918072248963.02124006454974.249980816
2248844.89589647455012.568086211
#Sta/Elev= 30
       0 2322.93       8 2317.56      20 2308.15      36 2294.47      48 2285.26
      60 2277.59      80 2267.73      84 2264.46      88 2259.64      92 2256.39
    94.7 2255.42     120 2254.65  137.792255.357   144.1 2256.78   168.1 2254.48
   180.1 2256.12   188.1 2255.37   220.1 2257.24   232.1  2254.7   244.1 2253.78
   256.1  2256.3   280.1 2255.13   308.1 2259.07   329.1 2257.72   337.5 2255.81
   366.9 2255.94   375.4 2259.13     388 2266.31   425.8 2294.52   433.5 2301.68
#Mann= 3 ,-1,0
       0      .1       0    94.7    .045       0  137.79      .1       0
Bank Sta=94.7,137.79
XS Rating Curve= 0 ,0
Exp/Cntr(USF)=0,0
Exp/Cntr=0.3,0.1

Type RM Length L Ch R = 1 ,5986    ,335.5,325,309.3
XS GIS Cut Line= 2
2249166.91920786454564.5934759882248738.54701453454804.899828346
#Sta/Elev= 30
       0 2292.27    16.9 2288.03    49.5 2282.62    58.3 2277.58    76.5 2260.51
    85.7 2253.06    93.5 2249.98   108.2 2248.76   143.1 2249.07   159.1 2251.58
   172.9 2251.06   184.6    2253   204.9 2253.45   218.7 2252.88   230.1 2250.89
   246.5  2250.7   262.8 2247.31   296.7 2248.59     308 2250.33   328.8 2248.18
     358 2249.68   396.2 2246.09   399.1  2246.5   406.8 2250.16   416.7  2249.1
   422.6 2249.64   438.9 2255.19   452.6 2268.64   466.4 2280.06   491.2 2305.19
#Mann= 3 ,-1,0
       0      .1       0   108.2    .045       0   143.1      .1       0
Bank Sta=108.2,143.1
XS Rating Curve= 0 ,0
Exp/Cntr(USF)=0,0
Exp/Cntr=0.3,0.1

Type RM Length L Ch R = 1 ,5661    ,297.2,298.1,295.8
XS GIS Cut Line= 2
2248878.47185259454322.9933359712248643.38955137454683.452864506
#Sta/Elev= 30
       0 2282.15    12.2 2280.13    16.9 2277.69    26.2 2269.42      36  2259.8
    45.6 2252.78    50.4 2250.36    69.5 2248.93    98.6 2248.31   102.9 2247.64
   112.4  2242.9     142 2242.75   150.6 2244.69     165 2245.15   184.1 2243.38
   201.9 2243.03   208.5 2241.18   231.8  2243.3   269.2 2242.97   292.3 2241.54
   298.7 2241.89   311.7  2244.1   321.2 2244.68   332.1 2247.34   341.4 2245.79
   347.2  2246.5   355.7 2250.35     363 2255.05   421.6 2301.53   430.3 2307.91
#Mann= 3 ,-1,0
       0      .1       0   112.4    .045       0     142      .1       0
Bank Sta=112.4,142
XS Rating Curve= 0 ,0
Exp/Cntr(USF)=0,0
Exp/Cntr=0.3,0.1

Type RM Length L Ch R = 1 ,5363    ,279.2,281.9,283.7
XS GIS Cut Line= 3
2248694.87570378454180.8931090812248615.88805057454217.565948072
2248439.57632466 454485.55977146
#Sta/Elev= 30
       0  2271.6    38.4 2268.72    53.4 2264.67    65.5  2262.9    69.1 2261.51
    82.4 2253.14    98.2 2246.23   105.8 2241.11   109.7 2239.71   124.9 2238.19
   137.5 2239.73   161.7 2241.01   193.5 2241.15   216.6  2240.3   230.3 2237.98
   242.6 2237.29   268.5 2237.28     283 2237.94   311.7 2235.16   321.2 2238.83
   332.1 2241.02     335 2242.66   337.9 2245.24     361 2268.04   375.4 2283.61
   378.3 2287.79   384.1 2300.36   388.3 2306.26   398.5 2316.03   407.9 2323.66
#Mann= 3 ,-1,0
       0      .1       0   242.6    .045       0   268.5      .1       0
Bank Sta=242.6,268.5
XS Rating Curve= 0 ,0
Exp/Cntr(USF)=0,0
Exp/Cntr=0.3,0.1

Type RM Length L Ch R = 1 ,5081    ,228.6,215.8,205.7
XS GIS Cut Line= 4
2248416.28337214 453985.140577862248344.13229211454141.464044845
2248274.00917529 454224.856022762248235.53368929454318.772179529
#Sta/Elev= 30
       0 2265.75    13.3 2253.18    17.7  2250.9    22.1 2250.01    26.5 2248.15
    30.9  2245.3    36.3 2242.82    78.5 2241.27    92.6 2239.49   110.2 2239.45
   124.3 2236.95   133.9 2236.32   153.8 2236.21   174.8 2237.06   192.7 2234.68
   209.4 2233.92   234.3 2231.05   251.4 2230.89   259.1  2230.7   265.9 2230.83
   277.8  2234.3   285.8 2234.68   294.4 2233.32   298.8 2233.44   307.4 2235.66
   316.1 2235.91   319.6 2236.91   324.7 2240.75   334.9 2249.93   382.6  2280.4
#Mann= 3 ,-1,0
       0      .1       0   234.3    .045       0   251.4      .1       0
Bank Sta=234.3,251.4
XS Rating Curve= 0 ,0
Exp/Cntr(USF)=0,0
Exp/Cntr=0.3,0.1

Type RM Length L Ch R = 1 ,4866    ,198.6,196.2,194.1
XS GIS Cut Line= 3
2248150.42509416453855.0690395932248082.72139141454247.186318025
2248103.87879852454306.427057932
#Sta/Elev= 30
       0 2272.38    14.3 2270.26    22.4 2266.09    58.7 2236.32    67.1 2232.14
    86.8 2230.89   119.9  2233.9   148.3 2229.59   164.5 2231.38   180.7 2231.38
   192.9 2232.98   217.3  2233.5   221.3  2232.4   229.5 2227.37   232.2 2226.88
   249.5 2226.41   259.9 2226.91   259.9 2226.92     270 2230.09   277.2 2231.17
   318.8 2231.53   330.9 2230.65   339.1  2228.3   353.4 2232.83   371.5 2232.71
   379.6  2233.6   391.5 2237.66   416.3 2250.41   438.5 2263.95   460.8 2279.65
#Mann= 3 ,-1,0
       0      .1       0   232.2    .045       0   259.9      .1       0
#XS Ineff= 2 , 0
          121.99  2251.5  356.93          2242.5
Permanent Ineff=
       F       F
Bank Sta=232.2,259.9
XS Rating Curve= 0 ,0
Exp/Cntr(USF)=0,0
Exp/Cntr=0.3,0.1

Type RM Length L Ch R = 1 ,4669    ,376.7,362.8,349
XS GIS Cut Line= 4
2247923.47034603453814.7861938112247922.96664846453958.302684347
2247900.90913714454246.5373733372247956.96648426454337.443393183
#Sta/Elev= 30
       0 2263.69    14.4 2251.55    26.4 2243.15    42.4 2230.34    46.4 2228.86
    58.4 2226.68    66.4 2226.17    94.4 2228.25   122.4 2228.71   146.4 2231.26
   170.5  2228.8   187.1 2229.93   204.7 2227.66   234.7 2229.64   242.7 2228.41
   252.2 2225.71   274.8 2225.09   283.62225.623   294.8  2227.8   322.9 2227.19
     343 2229.83   391.1 2229.81   407.2 2229.02   431.2 2230.57     463 2229.71
   473.3 2231.04   483.4 2234.79   499.8 2244.04     525 2262.96   539.4 2272.89
#Mann= 3 ,0,0
       0      .1       0   252.2    .045       0   283.6      .1       0
#XS Ineff= 2 , 0
                          431.36         2232.98
Permanent Ineff=
       F       F
Bank Sta=252.2,283.6
XS Rating Curve= 0 ,0
Exp/Cntr(USF)=0,0
Exp/Cntr=0.3,0.1

Type RM Length L Ch R = 1 ,4307    ,282.7,282.6,282.9
XS GIS Cut Line= 2
2247504.41893041454014.4548398192247749.84485289454439.013475819
#Sta/Elev= 30
       0 2283.12    12.4 2276.25    39.5 2258.43    72.5 2231.95    81.7 2222.87
    86.3 2219.85    95.4 2219.16   111.4 2219.54   118.7 2221.86   121.9 2222.22
   148.2 2221.57   174.1 2223.22   192.6 2222.02   197.2 2221.25   201.8 2219.62
   207.3    2219   224.3 2219.39   234.2 2221.86   243.4 2222.61   253.6 2225.04
   262.4 2226.15   282.9 2227.09   312.7 2225.99   382.4 2225.87   408.8 2226.66
   429.3 2228.02   438.1 2229.51   452.7 2234.36   479.1 2246.42   490.4 2252.62
#Mann= 3 ,-1,0
       0      .1       0    86.3    .045       0   111.4      .1       0
Bank Sta=86.3,111.4
XS Rating Curve= 0 ,0
Exp/Cntr(USF)=0,0
Exp/Cntr=0.3,0.1

Type RM Length L Ch R = 1 ,4024    ,223.8,231.5,239.3
XS GIS Cut Line= 2
2247257.83161608454153.8051880372247501.84704474454568.490367386
#Sta/Elev= 30
       0 2289.79     8.6 2282.36    21.7 2269.76    36.2 2259.86    59.6 2239.08
    74.3 2228.54    88.9 2216.69    92.1 2215.21    96.7  2214.7   133.9 2214.64
   152.4 2217.29   184.9 2217.51   189.6 2217.07   203.5 2213.81   217.2  2213.5
     222 2213.81     235 2219.29   240.6 2220.09     273    2220   290.5 2219.01
   305.6 2219.62   319.5 2221.96     328 2222.58   370.6 2220.44   375.2 2220.78
   407.4 2231.92     417 2233.35     454 2241.37     470 2246.33   481.2  2250.6
#Mann= 3 ,0,0
       0      .1       0    96.7    .045       0   133.9      .1       0
#XS Ineff= 2 , 0
                          241.46         2231.62
Permanent Ineff=
       F       F
Bank Sta=96.7,133.9
XS Rating Curve= 0 ,0
Exp/Cntr(USF)=0,0
Exp/Cntr=0.3,0.1

Type RM Length L Ch R = 1 ,3792    ,197.5,201.7,204.5
XS GIS Cut Line= 2
2247071.39733157454214.7449604572247184.23683615454671.744954025
#Sta/Elev= 30
       0 2272.21    27.2 2250.41    43.7 2240.08    60.2 2227.99    75.3 2218.75
    80.8 2216.62    88.6 2215.22    98.5 2211.51   108.4 2210.73     122 2210.29
   131.5 2210.92   138.5 2212.24   159.1 2212.62   196.2 2211.58   204.4 2214.06
   210.8 2214.91   220.9 2214.82   233.2 2212.09   241.5  2213.4   274.4 2215.18
   290.9 2215.42   311.5  2213.9   336.4 2215.94   352.7 2215.64   369.2 2216.68
   377.4 2218.86   403.7 2230.94   418.6 2234.25   447.5 2244.26   470.7 2253.32
#Mann= 3 ,-1,0
       0      .1       0   108.4    .045       0   131.5      .1       0
#XS Ineff= 2 , 0
                          287.15         2229.77
Permanent Ineff=
       F       F
Bank Sta=108.4,131.5
XS Rating Curve= 0 ,0
Exp/Cntr(USF)=0,0
Exp/Cntr=0.3,0.1

Type RM Length L Ch R = 1 ,3591    ,322.4,318.4,326.3
XS GIS Cut Line= 3
2246962.84432297454204.4252279762246896.52278524 454300.79871249
2246934.86492424454708.054405114
#Sta/Elev= 30
       0 2268.67    11.8 2262.56      64 2231.38    75.3  2226.3    85.9  2222.9
     106 2218.02   133.4 2213.49   145.5 2210.49   161.1  2208.6   195.62208.653
   205.8 2208.06   217.8 2209.72   241.9 2210.72     262 2208.22   278.6 2211.58
   326.3 2209.75   334.3 2211.42   348.4 2211.87   358.4 2211.97   370.5 2210.03
   378.5 2211.57   406.6 2209.93   414.7 2210.91   430.8 2211.35   434.8  2212.7
   438.8 2215.47   466.9 2237.44   474.9 2241.31   503.1 2252.05     526 2262.03
#Mann= 3 ,0,0
       0      .1       0   161.1    .045       0   195.6      .1       0
Bank Sta=161.1,195.6
XS Rating Curve= 0 ,0
Exp/Cntr(USF)=0,0
Exp/Cntr=0.3,0.1
